HEC-RAS study PPO_Kvasiny_efektiv.prj: PPO_Kvasiny_efektivita

--- PPO_Kvasiny_efektiv.g01 (geometry) --- (continued)

Type RM Length L Ch R = 1 ,16947.94,14.61,14.1,13.66
XS GIS Cut Line= 6
    -610169.5517   -1045485.6161-610173.24989999    -1045477.427
    -610183.6554   -1045466.7471-610201.92269999   -1045457.7056
    -610218.8174   -1045438.1758    -610302.8072   -1045298.9794
#Sta/Elev= 30
       0  356.32    4.38  352.23    6.07  350.95    6.77  350.22   19.78  349.49
   22.82  349.66    23.9  349.91   28.73  349.91   28.74  348.84   29.13  348.41
   30.46  347.61   37.39  347.77   38.04  348.04   40.11  349.42   48.72  349.64
   59.87  349.69   61.96  349.79   64.59  350.12   76.11  349.83  109.33  349.71
  119.86  349.78  172.83  349.51  185.94  349.61  197.09  349.42   222.4  349.38
  222.92   348.8   224.5   348.8  227.52  350.97  228.79  352.13  232.67  354.58
#Mann= 3 , 0 , 0
       0      .1       0   28.73    .045       0   40.11     .09       0
Levee=0,,,-1,40.75,350.9502,,	2158
Bank Sta=28.73,40.11
XS Rating Curve= 0 ,0
Exp/Cntr=0.3,0.1

Type RM Length L Ch R = 1 ,16933.84,27.14,24.89,15.43
XS GIS Cut Line= 6
    -610172.8312   -1045503.2958    -610183.6262   -1045487.4208
    -610192.1378   -1045478.4949    -610208.3665   -1045469.9668
    -610228.7441   -1045448.1827    -610312.5439   -1045301.5194
#Sta/Elev= 30
       0  364.96    6.16   364.6    8.34  362.41   19.24  349.88   21.81   349.6
   31.53  350.04   32.63  349.98   36.25  347.68   43.98  347.81    44.6  348.34
    46.6  349.24   47.05  349.28      74  349.63   76.83     350   82.89  349.84
    88.8  349.51   99.14  349.54  105.83  349.75  137.71  349.66  141.24  349.75
  173.25  349.39  218.78  349.42  227.56  349.21  235.14  349.26  235.67  348.69
  237.01  348.69  239.77  351.08  241.66  352.51   246.9  355.87  248.61  356.83
#Mann= 3 , 0 , 0
       0      .1       0   32.63     .05       0   47.05      .1       0
Levee=0,,,-1,46.74,350.7523,,	2158
#Block Obstruct= 2 ,-1
   54.52   58.56352.4616   62.43   72.37352.5712
Bank Sta=32.63,47.05
XS Rating Curve= 0 ,0
Exp/Cntr=0.3,0.1

Type RM Length L Ch R = 1 ,16821.12,43.01,41.79,41.65
XS GIS Cut Line= 2
-610275.27459999   -1045565.3143    -610395.3498   -1045343.0538
#Sta/Elev= 30
       0  361.46    3.71  360.82    6.05  360.65   17.33  360.98   20.94  358.62
   29.19  350.56   32.12   349.4   34.27  348.04   34.85  346.74   38.31  346.66
   41.55  346.67   43.58  348.44   54.15  348.27   66.86   348.4   93.44  349.04
  108.69  349.14  142.41  348.97  161.72  349.11  168.37  349.38   169.6  348.98
  171.36  348.92  202.82  348.56  212.54  348.64  214.81  348.83  229.46  348.84
  232.68  349.89   235.9  350.15  236.56  349.58  242.45  352.12  252.62  359.44
#Mann= 3 , 0 , 0
       0     .05       0   32.12     .05       0   43.58     .05       0
Levee=0,,,-1,44.24,349.9477,,	2158
#Block Obstruct= 1 ,-1
   53.58   64.61351.3344
Bank Sta=32.12,43.58
XS Rating Curve= 0 ,0
Exp/Cntr=0.3,0.1

Type RM Length L Ch R = 1 ,16751.94,21.77,21.42,20.49
XS GIS Cut Line= 3
-610331.99179999   -1045606.3583     -610368.002   -1045538.7669
    -610450.4891    -1045381.048
#Sta/Elev= 30
       0  359.83    3.86  359.16    7.68  358.91    13.1  358.87   13.71  358.77
   21.76  358.45   26.44  358.34   26.69  358.03   36.22     352   37.03  351.14
    39.3   349.4    43.3  346.47   46.95  346.38   51.43  346.62   53.67  347.82
   55.59  347.96   63.34  348.27    84.5   348.4  103.36  348.42  119.61  348.07
  137.55  348.17  154.31  348.46  188.11   348.8   214.3  348.57  232.32  348.69
   236.5  348.74  249.53  349.21  250.98  349.63  251.15  350.05  254.57  349.95
#Mann= 3 , 0 , 0
       0      .1       0    39.3     .05       0   55.59      .1       0
Levee=0,,,-1,56,349.5115,,	2158
#Block Obstruct= 2 ,-1
  184.93  199.08351.7553   56.68   63.33351.1675
Bank Sta=39.3,55.59
XS Rating Curve= 0 ,0
Exp/Cntr=0.3,0.1

Type RM Length L Ch R = 1 ,16730.52,4.86,4.82,4.85
XS GIS Cut Line= 3
    -610352.6812   -1045617.9347-610388.15709999   -1045543.0952
    -610465.3939   -1045389.8634
#Sta/Elev= 30
       0  358.93    9.19  357.93   14.08  358.21   22.01  357.45   27.93  354.09
   32.64  353.17   38.18  349.89   41.39  348.74   42.75  348.86   43.07   348.4
   43.43   346.9   44.17  346.39   48.14  346.29   52.25  346.36   53.34  346.67
   53.78  347.08   55.17  347.83   55.83  348.02   68.85  348.23    86.3  347.93
   97.54  348.18  109.47  347.99  142.98  348.11   148.1  348.02  181.48  348.75
  216.45  348.58  235.97  348.67  252.59  348.92  253.94  350.02  254.42  350.01
#Mann= 3 , 0 , 0
       0      .1       0   42.75     .05       0   55.83      .1       0
Levee=0,,,-1,56.44,349.5195,,	2158
#Block Obstruct= 2 ,-1
       0    8.43361.4715   58.22   64.91351.0959
Bank Sta=42.75,55.83
XS Rating Curve= 0 ,0
Exp/Cntr=0.3,0.1

Type RM Length L Ch R = 1 ,16725.7 ,12.99,14.15,15.54
XS GIS Cut Line= 3
-610357.07759999   -1045619.9076    -610392.5535   -1045545.0681
    -610471.4441   -1045388.2447
#Sta/Elev= 30
       0  358.73    8.25  357.95   13.74   358.1   21.33  357.43   25.38  355.29
   29.98  354.13   33.21  352.97   34.21  352.29   38.23  350.14   41.28  348.17
   43.17  347.33   43.48  346.77    43.9  346.24   52.08  346.36   53.19  346.68
   55.07  347.84   56.99  347.96   65.11  348.18   84.43  347.85   95.58  348.09
  108.04  347.88  116.51  348.04   141.6  348.08  150.14  347.93  185.69   348.8
  222.57  348.62  252.83     349  253.56  349.11  256.38     350  258.37  350.05
#Mann= 3 , 0 , 0
       0      .1       0   41.28     .05       0   56.99      .1       0
Levee=0,,,-1,54.48,348.9688,,	2161
#Block Obstruct= 1 ,-1
       0    8.03361.3521
Bank Sta=41.28,56.99
XS Rating Curve= 0 ,0
Exp/Cntr=0.3,0.1

Type RM Length L Ch R = 1 ,16711.55,25.25,25.95,28.78
XS GIS Cut Line= 6
-610364.63259999   -1045627.0364    -610377.2875   -1045602.5042
-610393.99859999   -1045577.0942    -610395.3159   -1045574.2261
    -610401.3596   -1045562.6079    -610487.1075   -1045395.4414
#Sta/Elev= 30
       0  358.55   11.42  357.93   16.23   357.9   24.38  356.88   26.34  356.18
   31.38  354.97   40.08  349.03   44.53  347.35   46.16  346.17   53.25  345.98
   54.11  345.99   55.32  347.27   55.84  347.68   61.13  347.85   74.22  347.97
   84.94  347.84   96.79  347.92  107.67  347.77  127.94  347.73  148.62  348.12
  162.19  348.01  181.37  348.38  198.87  348.18  216.75  348.32  224.73  348.14
  229.48  348.15   253.4  348.57  254.72  349.52  256.17   350.2  262.14  350.16
#Mann= 3 , 0 , 0
       0      .1       0   40.08     .05       0   55.84      .1       0
Levee=0,,,-1,57.02,349.237,,	2161
#Block Obstruct= 4 ,-1
   61.17   74.27350.9031  150.01  161.74351.0612  189.46  214.16351.2825
       0    10.6361.2628
Bank Sta=40.08,55.84
XS Rating Curve= 0 ,0
Exp/Cntr=0.3,0.1

Type RM Length L Ch R = 1 ,16685.61,17.06,18.42,16.35
XS GIS Cut Line= 3
-610382.98559999   -1045633.4457-610424.52349999    -1045581.395
-610511.87249999   -1045407.5064
#Sta/Elev= 30
       0   358.3    9.52  357.21   11.52   356.4    18.7  356.09   26.62  356.05
   35.31  348.56   39.94  346.03   47.87   345.7   49.47  347.74   52.52  347.37
   54.79  347.68   91.59  347.51  107.49  347.93   116.4  347.55  124.24  347.58
  132.27  347.37  135.69  348.04  149.62  348.01  152.87  347.58   158.1  347.84
  174.46  348.06  205.73  348.08  228.44  347.88  241.77  348.03  250.63  348.37
  253.06  349.83  256.27  349.87   257.4  349.02  259.08  349.02  261.19  349.98
#Mann= 3 , 0 , 0
       0      .1       0   35.31     .05       0   49.47      .2       0
Levee=0,,,-1,50.97,348.9799,,	2161
#Block Obstruct= 5 ,-1
    56.1   62.64350.6454   52.52    56.1350.4926  148.46  160.19350.9218
  116.67  126.02350.5445  244.02  248.89351.2354
Bank Sta=35.31,49.47
XS Rating Curve= 0 ,0
Exp/Cntr=0.3,0.1

Type RM Length L Ch R = 1 ,16667.18,6.2,5.78,6.81
XS GIS Cut Line= 4
    -610393.8158    -1045643.949-610416.82609999   -1045617.2862
    -610427.9386   -1045608.2904-610522.61459999   -1045420.9473
#Sta/Elev= 30
       0  358.13    9.83  357.15   12.01  355.97   23.98  355.89   33.56  349.97
   35.22   348.7   38.62  346.02   40.35  345.83   46.29  345.68      48  347.55
   58.83  347.66   64.61  347.93   73.46  347.62   92.26  347.44   92.35  347.33
  101.51  347.59  108.59  347.46  113.83  347.53   120.2  347.29  147.91  347.45
  158.38  347.25   170.8   347.9  205.99  347.86  232.66  347.54  233.67  348.07
  243.08  347.93  254.22  348.12  254.91   348.2  257.28   349.9  259.42  349.93
#Mann= 3 , 0 , 0
       0      .1       0   35.22     .05       0      48      .2       0
Levee=0,,,-1,51.6,349.0984,,	2161
#Block Obstruct= 3 ,-1
   58.83   65.46350.7798  190.67  201.55350.8297  240.54   248.8 350.981
Bank Sta=35.22,48
XS Rating Curve= 0 ,0
Exp/Cntr=0.3,0.1

Type RM Length L Ch R = 1 ,16661.4 ,5.64,6.86,5.9
XS GIS Cut Line= 6
    -610396.1494   -1045646.1225-610420.53339999   -1045622.2464
-610432.85249999   -1045611.3244    -610443.2665   -1045593.5444
-610481.36659999   -1045517.8522    -610525.4721   -1045423.9106
#Sta/Elev= 30
       0  358.16    9.91  357.17   11.97  355.84   22.33  355.74   23.87  354.91
   34.35  348.36   37.29  346.05   39.09  345.81   42.58  345.74   45.69  345.75
   47.63  347.64   60.93  347.61   65.96  347.73   88.16  347.46   91.18  347.38
    91.3  347.23  102.31  347.47  104.31  347.27  115.28     347  131.44  347.12
  143.54   347.5  157.87  347.21  161.14  347.27   172.1  347.93  234.14   347.5
  235.04   348.1  239.62  347.98  256.23  348.23  258.71  349.95  259.72  350.01
#Mann= 3 , 0 , 0
       0      .1       0   34.35     .05       0   47.63      .2       0
Levee=0,,,-1,54.42,349.1576,,	2161
#Block Obstruct= 2 ,-1
  192.18  203.07350.7415  242.01  250.28351.0749
Bank Sta=34.35,47.63
XS Rating Curve= 0 ,0
Exp/Cntr=0.3,0.1

Type RM Length L Ch R = 1 ,16654.54,6.93,6.66,6.8
XS GIS Cut Line= 6
     -610399.919   -1045646.2163-610414.10069999   -1045633.6221
    -610423.8823   -1045626.7642    -610435.5652   -1045618.9463
    -610478.4107   -1045542.1985    -610530.1288   -1045427.2973
#Sta/Elev= 30
       0  357.92    7.45  357.15    9.46  355.71   18.93  355.45   20.83  354.18
   25.96  351.25   30.91  348.08   33.84  346.09   35.52  345.79   42.23  345.62
   44.97  347.61   45.65  347.71    64.5  347.61   74.01  347.38   83.87   347.4
   91.33  347.28   91.45  347.14  101.75  347.37  118.19  346.84  124.78  346.83
  142.08  346.87  143.13   347.4  163.07  347.62  170.12  347.96  171.35  347.84
  189.38  347.64  234.41  347.52  235.09  348.07  255.59  348.27  258.87  350.02
#Mann= 3 , 0 , 0
       0      .1       0   30.91     .05       0   45.65      .2       0
Levee=0,,,-1,55.88,349.1129,,	2161
#Block Obstruct= 3 ,-1
  241.83  250.11351.1296  192.08  202.98 350.625  107.84  132.87350.0207
Bank Sta=30.91,45.65
XS Rating Curve= 0 ,0
Exp/Cntr=0.3,0.1

Type RM Length L Ch R = 1 ,16647.88,5.99,6.32,7.53
XS GIS Cut Line= 6
-610407.45239999   -1045648.6625    -610428.5344   -1045631.8985
-610441.36149999   -1045622.7545-610461.68149999   -1045585.1624
    -610491.7806   -1045526.1073-610535.63219999   -1045432.9065
#Sta/Elev= 30
       0  357.49    4.15  357.11    6.59  355.39   15.07  355.31   25.93   347.9
   28.84  346.08   30.75  345.72   34.39  345.65   37.38  345.68   40.85  347.88
   44.05  347.89   46.97  346.75   51.41  346.92   71.69  346.83   79.54  347.25
   88.55  347.23   90.11  347.05   99.78  347.29  117.27  346.75  137.81  346.85
  140.96  346.93  141.89   347.4  146.14  347.36  165.71  348.02  166.93   347.6
  170.19  347.78  231.94  347.44  233.44  347.99  252.59  348.38   254.7  349.31
#Mann= 3 , 0 , 0
       0      .1       0   25.93     .05       0   40.85      .2       0
Levee=0,,,-1,76.74,348.5952,,	2159
#XS Ineff= 2 , 0
                           42.41          347.69
Permanent Ineff=
       F       F
#Block Obstruct= 3 ,-1
  105.66  130.77  349.98  190.35  201.24350.5325  239.91  248.18351.2398
Bank Sta=25.93,40.85
XS Rating Curve= 0 ,0
Exp/Cntr=0.3,0.1

Type RM Length L Ch R = 1 ,16641.56,17.07,15.6,12.26
XS GIS Cut Line= 6
-610413.30689999   -1045653.7066-610431.29479999   -1045637.3368
-610446.09189999    -1045627.568    -610459.5562   -1045605.4465
    -610472.0445   -1045581.5282    -610537.3255   -1045444.4423
#Sta/Elev= 30
       0   357.4    3.78     357    5.96  354.94   14.03  354.64   22.68  349.09
    26.9  346.03   28.84  345.65   31.89  345.59   35.63  345.75   39.44  348.15
   42.05  348.16   45.25  346.88   73.49  346.81   83.79  347.42   84.32  347.08
   92.09  346.97   100.1  347.18  120.88  346.64  140.97  346.88  143.73  347.19
  149.61  347.23  164.14  348.01  164.93  348.62  169.11  348.42  170.12  347.86
  176.98  347.58  205.67  347.42  233.34  347.37  234.95  347.94  246.77   348.2
#Mann= 3 , 0 , 0
       0      .1       0   22.68     .05       0   39.44      .1       0
Levee=0,,,-1,84.49,348.5743,,	2159
#XS Ineff= 2 , 0
                           41.88           347.8
Permanent Ineff=
       F       F
#Block Obstruct= 3 ,-1
   79.31   84.32350.0773  191.83  202.72350.4694  241.25  246.77351.1385
Bank Sta=22.68,39.44
XS Rating Curve= 0 ,0
Exp/Cntr=0.3,0.1

Type RM Length L Ch R = 1 ,16625.96,21.61,20.6,17.48
XS GIS Cut Line= 6
-610425.68789999   -1045669.8678     -610440.574   -1045651.9392
-610455.03269999   -1045638.1208     -610482.421   -1045587.8698
    -610520.3187      -1045502.6-610545.36879999   -1045446.8765
#Sta/Elev= 30
       0   357.1    4.18  356.86    6.41  356.35   10.26  353.98   18.26  353.74
   25.94  348.99   27.45  347.91   29.46  345.68   33.12  345.48   36.79  345.73
   42.22  348.16   44.24  348.13   47.11  346.82   80.33  346.76   85.96  347.12
   99.43  346.84  106.46  347.03   123.8  346.54   143.2  346.57  147.34  346.86
  147.63  347.45  149.17  348.39  150.21  348.33  154.14  346.76  154.35  348.03
  180.32  347.32  229.76  347.32  239.84  347.37  241.88  347.87  254.94  348.08
#Mann= 3 , 0 , 0
       0      .1       0   25.94     .05       0   42.22     .08       0
Levee=0,,,-1,91.1,348.5402,,	2159
#XS Ineff= 2 , 0
                           43.59          347.69
Permanent Ineff=
       F       F
#Block Obstruct= 3 ,-1
     113  124.22349.5901  198.32  209.22350.3801  247.62  254.94350.9503
Bank Sta=25.94,42.22
XS Rating Curve= 0 ,0
Exp/Cntr=0.3,0.1

Type RM Length L Ch R = 1 ,16605.36,21.02,20.3,16.27
XS GIS Cut Line= 3
-610445.09629999   -1045684.5852-610473.44709999   -1045644.2738
-610552.67139999    -1045460.529
#Sta/Elev= 30
       0  356.58     .55  356.59    2.78  355.95    5.88  354.21   11.21  354.03
   12.46  353.49   19.13  352.84   27.91  348.11   30.05  345.45   33.32  345.37
   38.15  345.73   42.18  347.67   43.48  347.65   46.26  346.67   84.14  346.69
   87.53     347  103.21   346.7  109.51  346.86  111.41  346.66  122.47  346.42
  139.16  346.36   144.1  346.64  156.37  346.35  158.08  348.05  176.45  347.81
  198.52  347.26  222.94   347.2  242.73  347.21  244.96  347.81  249.38  347.93
#Mann= 3 , 0 , 0
       0      .1       0   27.91     .05       0   42.18      .1       0
Levee=0,,,-1,94.36,348.3709,,	2159
#XS Ineff= 2 , 0
                           42.87          347.36
Permanent Ineff=
       F       F
#Block Obstruct= 3 ,-1
   89.25   94.26349.9202  138.07  142.43349.4565  201.36  212.27350.2634
Bank Sta=27.91,42.18
XS Rating Curve= 0 ,0
Exp/Cntr=0.3,0.1

Type RM Length L Ch R = 1 ,16585.06,17.86,16.08,10.48
XS GIS Cut Line= 4
    -610464.0819   -1045699.0756    -610487.7346   -1045656.9739
    -610509.9596   -1045590.2987    -610560.0797   -1045465.2915
#Sta/Elev= 30
       0  356.87    7.92  356.19   13.39  352.95   15.62  352.55   24.98  352.17
   25.73  351.56   26.49  351.16    31.3  347.03   33.63  345.24   36.97  345.18
   39.85  345.24   43.72  347.03   44.65  347.06   45.84  346.65   49.93   346.5
   93.75  346.75  107.37  346.59  113.82  346.71  118.99  346.34  122.48  346.25
  137.76  346.25  157.18  346.38  158.11  346.51  170.11  346.62  183.44  347.03
  196.43  347.18  231.58  347.31  247.21  347.17  249.92  347.78  253.25  347.81
#Mann= 3 , 0 , 0
       0      .1       0    31.3     .05       0   43.72      .1       0
Levee=0,,,-1,99.07,348.1866,,	2159
#XS Ineff= 2 , 0
                           43.98          346.83
Permanent Ineff=
       F       F
#Block Obstruct= 3 ,-1
  122.33  133.19349.2643  157.26  167.42349.4925  223.47  232.02350.2849
Bank Sta=31.3,43.72
XS Rating Curve= 0 ,0
Exp/Cntr=0.3,0.1

Type RM Length L Ch R = 1 ,16568.98,14.3,13.1,11.02
XS GIS Cut Line= 5
    -610486.8255   -1045706.5634-610495.14299999   -1045679.7281
    -610497.7888   -1045668.0863    -610514.7221    -1045594.532
    -610561.2439   -1045478.4149
#Sta/Elev= 29
       0  355.37    2.76  355.32    7.58  354.77   12.03  353.94   15.54  352.49
   22.92  351.99   26.09  351.85   28.89   348.7   28.92  348.54   29.95  345.51
   31.19  345.23   34.85  345.03   38.95   345.1   39.31  345.75   39.49  345.96
   42.33  346.09   43.66  346.22   51.97  346.48   78.74  346.53   91.89  346.67
  105.62  346.54  112.26  346.63  118.88   346.2  136.17  346.19     171  346.62
  184.22  347.01  200.78  347.12  212.99  347.32   240.6  347.21
#Mann= 3 , 0 , 0
       0      .1       0   28.92     .05       0   42.33      .1       0
Levee=0,,,-1,97.59,348.1275,,	2159
#Block Obstruct= 3 ,-1
    3.69   15.95356.8368  155.62  173.94 349.579  223.92   240.6350.2427
Bank Sta=28.92,42.33
XS Rating Curve= 0 ,0
Exp/Cntr=0.3,0.1

Type RM Length L Ch R = 1 ,16555.88,20.77,21.27,17.9
XS GIS Cut Line= 5
    -610504.2404   -1045706.1507    -610509.2146    -1045681.174
    -610509.4305   -1045668.0863-610521.60139999   -1045611.4654
    -610562.8314   -1045479.6849
#Sta/Elev= 27
       0  354.23   13.02  351.99   23.42  351.61   24.51  350.56   27.39  346.81
   27.78  345.31   29.57  345.03   30.58  344.97   34.36  344.97    35.5  345.15
   37.44  346.06   49.54  346.46    66.5   346.5   78.34  346.15   87.71  346.45
    94.9  346.37   105.3  346.49  108.23  346.24  136.11  346.09  150.44  346.55
  166.72  346.63  179.56  347.01  199.26  347.17  211.42  347.19  215.11  347.13
  228.36  347.25  234.55  347.19
#Mann= 3 , 0 , 0
       0      .1       0   27.39     .05       0   37.44      .1       0
Levee=0,,,-1,91.29,347.9076,,	2159
#Block Obstruct= 4 ,-1
       0   12.06356.1919  114.23   127.2349.1687  162.31  167.39349.6144
  228.72  234.55350.2217
Bank Sta=27.39,37.44
XS Rating Curve= 0 ,0
Exp/Cntr=0.3,0.1

Type RM Length L Ch R = 1 ,16534.61,4.61,4.56,4.51
XS GIS Cut Line= 6
-610529.54529999   -1045705.4184    -610529.8783    -1045676.323
-610530.17399999   -1045665.9981-610534.91189999   -1045624.3717
-610542.27789999   -1045575.2226-610569.46539999   -1045481.1129
#Sta/Elev= 30
       0  352.96   10.36  351.82   11.14   351.5   23.66  351.98   25.57  349.56
   30.35   347.5   30.86  346.87   31.51  345.46   32.53  344.46   33.67  344.45
   33.87  344.25   34.87  344.25   35.07  344.45   38.74  344.44   38.94  346.29
   39.07  346.31   42.57  346.46   81.81  345.97    82.6  346.22   86.73  346.17
   89.08  346.31   96.62   346.2  131.61  346.14  145.25  346.64  158.29  346.74
  169.44  346.98  193.45  346.81   208.9  346.89  224.82  347.13  228.98  347.35
#Mann= 3 , 0 , 0
       0      .1       0   30.86     .04       0   39.07      .1       0
Levee=0,,,-1,80.25,347.4962,,	2159
Bank Sta=30.86,39.07
XS Rating Curve= 0 ,0
Exp/Cntr=0.3,0.1

Type RM Length L Ch R = 1 ,16530.05,3.73,4.02,4.32
XS GIS Cut Line= 6
    -610534.1055   -1045705.0639-610534.43849999   -1045675.9685
    -610534.7342   -1045665.6436    -610539.4721   -1045624.0172
    -610546.8381   -1045574.8681    -610573.0214   -1045482.6369
#Sta/Elev= 30
       0  352.74    5.83  352.05    9.26  351.84   10.02  351.49   23.34  351.78
   24.68  349.86   27.24  348.46   30.35  346.97   30.99  346.81    31.1   345.7
   31.21  345.22   31.46  344.97   32.23  344.28   33.48  344.28   33.76  344.07
   34.69  344.07   34.89  344.27   38.61  344.26   38.85  346.33   43.12  346.47
   46.35  346.34   61.25  346.44   70.06  346.34   73.04  346.07   86.57  346.27
  127.43  346.18  155.85  346.84  208.55  346.82  224.39  347.06   226.9  347.24
#Mann= 3 , 0 , 0
       0      .1       0   30.99     .04       0   38.85      .1       0
Bank Sta=30.99,38.85
XS Rating Curve= 0 ,0
Exp/Cntr=0.3,0.1

Type RM Length L Ch R = 1 ,16526.03,4.58,4.2,3.62
XS GIS Cut Line= 5
    -610538.0693   -1045702.3362-610538.07229999    -1045677.112
    -610539.6568   -1045657.3569-610551.82759999   -1045576.9234
    -610578.2707   -1045483.1449
#Sta/Elev= 30
       0  352.26     5.9  351.85    6.62  351.49   20.62  351.63   21.48   350.4
   24.99  348.48    27.6  346.74   28.16  346.23   28.28  345.52   28.91  344.91
   29.51  344.13   31.02  344.12   31.22  343.92   32.08  343.91   32.44  344.11
   36.11  344.09   36.75  344.98   37.03  345.86    38.2  346.13   40.68  346.32
   57.07  346.33   66.05   346.3   70.55  346.04   81.67  346.21   96.26  346.06
  147.15  346.72  159.66  346.61   195.9   346.8  206.17  346.73  223.83  347.06
#Mann= 3 , 0 , 0
       0      .1       0   28.16     .04       0    38.2      .1       0
Bank Sta=28.16,38.2
XS Rating Curve= 0 ,0
Exp/Cntr=0.3,0.1

Type RM Length L Ch R = 1 ,16521.83,6.74,6.01,5.22
XS GIS Cut Line= 4
    -610542.1235   -1045699.3356    -610543.0548   -1045657.4255
    -610557.9562   -1045571.9967    -610579.7877   -1045484.1398
#Sta/Elev= 30
       0     352    2.23  351.87    2.87  351.49   17.63  351.46   17.91  351.07
    20.5  349.46   23.79  346.44    24.4  345.88   25.03   345.7   26.26  343.97
   28.45  343.96   28.64  343.76   28.85  343.75   29.66  343.75   29.86  343.95
   33.34  343.93   34.64  345.63   35.71  346.08   43.23   346.2    59.7  345.99
   62.86  346.11   67.39  345.99   76.82  346.17   84.53  346.16   85.58  346.05
   90.13  346.02   142.7  346.64  156.61  346.58  202.73  346.71  219.17  347.05
#Mann= 3 , 0 , 0
       0      .1       0   23.79     .04       0   35.71      .1       0
Bank Sta=23.79,35.71
XS Rating Curve= 0 ,0
Exp/Cntr=0.3,0.1

Type RM Length L Ch R = 1 ,16515.82,2.86,2.86,2.83
XS GIS Cut Line= 5
    -610549.2021   -1045701.0436    -610549.7798   -1045679.3474
    -610548.1328   -1045663.7179    -610550.4721   -1045643.0045
    -610581.5868   -1045484.5631
#Sta/Elev= 30
       0  352.19    2.75  352.14    2.76  351.49   13.52   351.4   18.86  351.14
   20.33  351.32   23.28   347.4   26.15  345.56   26.81  345.44   28.06  343.72
   30.97  343.72   31.17  343.52   32.17  343.52   32.37  343.72   35.83  343.72
    37.1  345.42   38.47  346.01   38.68  346.02   58.86  345.66   64.28   345.9
   72.41  345.93   76.19  346.13   84.83  346.12   87.61  345.96   99.59  346.08
  112.21  346.05  137.16  346.48  188.56  346.73  203.93   346.7  219.73  347.06
#Mann= 3 , 0 , 0
       0      .1       0   26.15     .04       0   38.68      .1       0
Levee=0,,,-1,40.99,345.99,,
#Block Obstruct= 2 ,-1
   85.71  103.01  349.05  114.98  124.12349.1804
Bank Sta=26.15,38.68
XS Rating Curve= 0 ,0
Exp/Cntr=0.3,0.1

Type RM Length L Ch R = 1 ,16401.95,1.88,1.88,1.88
XS GIS Cut Line= 6
    -610643.0462   -1045735.4757    -610657.9483   -1045686.2902
-610661.88529999   -1045666.6815-610664.87119999    -1045645.638
-610675.02239999   -1045602.4955-610708.26749999   -1045527.6306
#Sta/Elev= 30
       0  350.39    9.85  349.85   12.56  347.74   19.29   347.7   26.28     347
   27.32  346.82    28.7  345.85   38.33  345.26   50.16  345.27   51.22  344.63
    55.9  344.29   57.83  341.86   64.94  341.58   66.39  341.74   69.38  344.11
   93.96  344.66   95.97  344.35  103.63  344.41  128.62  345.51  130.57  344.79
  145.58  345.11  147.47  345.72  183.43  345.49  199.49  345.85  205.61  346.54
  211.97  349.07  212.55  348.24   214.3  348.24  216.33   349.4  218.88  350.17
#Mann= 3 ,-1 , 0
       0      .1       0   56.59     .04       0   68.65      .1       0
#Block Obstruct= 1 ,-1
  110.49  119.04347.9603
Bank Sta=55.9,69.38
XS Rating Curve= 0 ,0
Exp/Cntr=0.3,0.1

Type RM Length L Ch R = 1 ,16400.07,8.96,8.12,7.29
XS GIS Cut Line= 6
-610644.88569999   -1045735.8526-610659.78779999   -1045686.6671
    -610663.7248   -1045667.0584    -610666.7107   -1045646.0149
    -610676.8619   -1045602.8724     -610710.107   -1045528.0075
#Sta/Elev= 30
       0  350.37    9.13  349.84   12.04  347.59   18.73  347.62   26.84  346.95
    29.1  345.74   37.36  345.23    50.4   345.3    51.9  344.66    56.3  344.07
   56.81  343.73   57.32  342.42   57.79  341.88   65.38  341.61   66.46  341.73
   69.43  344.04   93.66  344.59  103.99  344.37  131.13   345.5  132.29  344.81
  144.17  345.17   150.8  345.76  183.97  345.49  199.64  345.86  204.96  346.52
  211.66  349.09  212.24  348.26  213.94  348.26  216.49  349.75  218.88  350.47
#Mann= 3 , 0 , 0
       0     .08       0    56.3     .04       0   69.43     .08       0
#Block Obstruct= 2 ,-1
  110.43  118.98347.8619  136.33  137.43347.9948
Bank Sta=56.3,69.43
XS Rating Curve= 0 ,0
Exp/Cntr=0.3,0.1

Type RM Length L Ch R = 1 ,16241.06,21.08,23.12,26.17
XS GIS Cut Line= 4
-610740.67799999   -1045794.9927    -610783.6451   -1045731.5412
-610794.63679999   -1045726.0454-610856.08969999   -1045561.6711
#Sta/Elev= 30
       0  350.39   13.77  349.23   15.54  348.29   20.49  348.31   27.36  344.24
   36.66  344.11   42.33  343.78   42.34  342.86   48.03  342.66   65.38  343.26
   66.37  343.09   77.59   342.6   79.07  341.68   80.26  340.12   86.76  340.23
   88.63  341.88  106.11  342.02  115.13  341.86  116.79  343.16  126.05   343.4
  127.44  342.88  138.01   343.6   153.9  344.22  169.78  344.52  175.28  344.58
  198.75  344.37  218.04   344.5  250.18  344.31  256.93  344.86  264.41  348.75
#Mann= 3 , 0 , 0
       0     .08       0   77.59     .04       0   88.63     .08       0
Bank Sta=77.59,88.63
XS Rating Curve= 0 ,0
Exp/Cntr=0.3,0.1

Type RM Length L Ch R = 1 ,16217.94,17.82,14.38,10.85
XS GIS Cut Line= 6
    -610749.3409   -1045804.8633    -610792.0326   -1045754.9198
    -610808.2784   -1045743.2547    -610827.6222   -1045711.1307
    -610872.3427   -1045570.3783    -610872.3427   -1045555.1515
#Sta/Elev= 30
       0  350.71    8.39  350.24   16.02  349.44   17.41  348.65   22.55   349.1
   29.09  344.06   35.38  343.78   36.67  342.67   54.49  342.53   61.05  342.87
   71.24  342.38   72.85  341.54   73.02  339.95    73.1  339.81   74.14  339.76
   79.78  340.35   81.77  341.63  120.46  341.46     123  343.05  134.37  343.11
  136.79  342.81  140.02  342.79  156.08  343.09  187.68  344.15  265.62  344.29
  270.54  344.82  280.67   349.3  281.02  348.59  282.12  348.58  286.12  350.23
#Mann= 3 ,-1 , 0
       0     .08       0   72.44     .04       0   81.72     .08       0
Levee=0,,,-1,97.34,341.97,,
Bank Sta=71.24,81.77
XS Rating Curve= 0 ,0
Exp/Cntr=0.3,0.1

Type RM Length L Ch R = 1 ,16203.55,16.98,16.59,13.12
XS GIS Cut Line= 5
    -610769.6559   -1045808.4823    -610808.1264   -1045763.0171
    -610815.1211   -1045751.5259    -610847.5962   -1045700.0653
    -610890.0638   -1045564.6689
#Sta/Elev= 30
       0  350.46    2.07   350.4    4.97  349.97    6.36  349.96    9.56  349.67
   12.09  349.11   18.75  344.19   19.58   344.1   27.59  344.03    28.1  342.77
   30.81  342.75   38.12  342.41   62.52  342.29   62.53  339.83   67.37  339.93
   72.94   341.9  103.27  341.27  112.63  341.76  114.61  343.04  128.88  342.86
  139.06  342.85  148.15  342.95  150.27  343.06  154.36  343.02  186.61  343.96
  255.33  344.14  264.57  344.44  268.36   344.8  270.82  345.96  275.76  348.03
#Mann= 3 , 0 , 0
       0     .08       0   62.52     .04       0   72.94     .08       0
Levee=0,,,-1,73.61,341.88,,
#Block Obstruct= 4 ,-1
  153.07  163.46346.1526       0    3.74353.3066   27.86   34.56 345.952
   39.28   51.69345.3915
Bank Sta=62.52,72.94
XS Rating Curve= 0 ,0
Exp/Cntr=0.3,0.1

Type RM Length L Ch R = 1 ,16186.97,23.06,21.77,16.29
XS GIS Cut Line= 5
    -610779.6482   -1045816.9759    -610825.1134   -1045768.5129
    -610828.6108   -1045757.0217-610860.08659999   -1045702.5634
    -610908.5496   -1045574.6612
#Sta/Elev= 30
       0  350.62    5.89  350.41   11.51  349.41    18.9  344.17   24.48  343.71
   26.19  342.77   31.27  342.48   43.49  342.32   66.78  342.22   68.32  341.18
   68.33  339.88   74.81  339.93   77.62  341.78   81.26   341.5  100.37  341.66
  104.66  341.62   114.7  342.03     117  342.24  118.59  343.04   132.6  342.82
  141.36  342.84  148.28  342.99  150.56   343.4  160.08  343.12  181.77  343.31
  197.52  343.81  205.12  343.88  261.78  343.81  276.45  344.65  278.14  345.52
#Mann= 3 , 0 , 0
       0     .08       0   66.78     .04       0   77.62     .08       0
Levee=0,,,-1,78.12,341.73,,
#Block Obstruct= 1 ,-1
       0    3.38 353.571
Bank Sta=66.78,77.62
XS Rating Curve= 0 ,0
Exp/Cntr=0.3,0.1

Type RM Length L Ch R = 1 ,16165.19,23.88,24.21,22.28
XS GIS Cut Line= 4
    -610790.1402   -1045840.9575-610846.59699999    -1045775.008
    -610849.0951   -1045761.5183-610919.04149999   -1045584.6535
#Sta/Elev= 27
       0   350.3    7.18  349.42   15.14  349.01   18.29  346.69   22.32   344.1
   28.64  343.85   31.14  343.22   44.85  342.19   50.01  341.93   67.73  341.81
   81.92   342.1   81.93  339.82   90.15  340.05   90.61  340.92   91.47  341.52
   91.57  341.52   94.87  341.37  119.58  341.76  130.35  342.66  141.45  342.89
  148.64  342.77  187.72  343.26  204.08   343.7  213.17  343.78  245.14  343.64
  277.62  343.76  283.46  344.16
#Mann= 3 , 0 , 0
       0     .08       0   81.92     .04       0   91.57     .08       0
Levee=0,,,-1,92.49,341.5,,
#Block Obstruct= 3 ,-1
   44.75   48.05345.5259   69.81   74.72344.8481  113.88  124.65344.7277
Bank Sta=81.92,91.57
XS Rating Curve= 0 ,0
Exp/Cntr=0.3,0.1

Type RM Length L Ch R = 1 ,16140.98,20.09,21.91,20.25
XS GIS Cut Line= 4
    -610811.1241   -1045849.9506    -610870.5786   -1045779.5045
-610873.07669999   -1045762.0179    -610940.0255   -1045585.6527
#Sta/Elev= 29
       0  349.09   13.38  348.34   19.31   344.1   20.29  343.83   22.43  343.57
   35.21  342.71   39.32  342.27   63.88  341.84   89.62   341.9   89.63  339.77
   96.74  339.89  100.43     341  110.58  341.06  122.46   342.2   137.9  342.79
  142.93  343.06  145.31  343.03  158.93  343.32  168.61  343.16  174.96  343.19
  192.29  343.56  206.78  343.74  223.24   343.5   239.2  343.55  255.24  343.34
  278.02  343.51   287.4   343.7  290.74  344.11  291.95  344.86
#Mann= 3 , 0 , 0
       0     .08       0   89.62     .04       0  100.43     .08       0
#Block Obstruct= 1 ,-1
   69.69   82.07344.8526
Bank Sta=89.62,100.43
XS Rating Curve= 0 ,0
Exp/Cntr=0.3,0.1

Type RM Length L Ch R = 1 ,16007.74,6.71,7.01,8.54
XS GIS Cut Line= 6
-610971.77129999   -1045859.4797    -610980.0408   -1045836.7296
    -610989.9356   -1045825.7279    -610992.9954   -1045818.0942
-611010.51089999   -1045778.8608    -611023.0044   -1045744.3002
#Sta/Elev= 29
       0  343.71    1.32  343.69    2.18  342.92    2.77   342.5    5.13  342.36
   12.14  341.72   18.24  341.46   25.68  341.27   26.28  340.69   27.86  339.54
    29.2     339   29.37  338.85   37.58  338.76   37.59  338.76   37.72  340.66
   37.91  340.87   39.28  341.03   47.07  341.11   50.26  341.06    60.7  341.44
   68.38  342.03   75.18  342.15   76.81  341.95   79.46  341.93   83.71  341.74
   89.23  341.72   98.01  341.84  114.86  342.26  126.94  342.35
#Mann= 3 , 0 , 0
       0     .08       0   25.68    .035       0   39.28      .1       0
Bank Sta=25.68,39.28
XS Rating Curve= 0 ,0
Exp/Cntr=0.3,0.1

Type RM Length L Ch R = 1 ,16000.73,9.83,10.81,10.61
XS GIS Cut Line= 5
     -610976.975   -1045864.1751    -610985.2445    -1045841.425
    -610997.4496   -1045827.8546-611019.62709999   -1045783.7506
    -611027.9807   -1045754.2729
#Sta/Elev= 26
       0  344.23     5.8  343.93    8.46   342.3    9.96  342.01   11.85  341.78
   18.91  341.45   27.28  341.26   27.95  341.12   28.78  338.98    29.1  338.72
   33.82  338.45   36.88  338.62   36.89   340.2   36.91  340.33   40.15  340.89
   50.35  340.93   53.21  340.83   60.15  341.08   63.25  341.08   65.41  341.56
   67.34  341.78   75.75  342.01   76.44  342.02   77.92  341.86   87.77  341.77
  122.46   342.2
#Mann= 3 , 0 , 0
       0      .1       0   27.28    .035       0   40.15     .08       0
Levee=0,,,-1,40.08,342.3748,,	2160
#Block Obstruct= 3 ,-1
       0    5.64347.0853    82.3  100.74344.8723   50.41   61.78343.9916
Bank Sta=27.28,40.15
XS Rating Curve= 0 ,0
Exp/Cntr=0.3,0.1

Type RM Length L Ch R = 1 ,15989.93,23.84,22.47,19.81
XS GIS Cut Line= 6
    -610970.3973   -1045887.0677    -610993.4662   -1045848.7396
    -611005.6395   -1045834.6026    -611029.7291    -1045788.774
    -611034.3488   -1045770.0031    -611035.9998    -1045753.747
#Sta/Elev= 30
       0  346.39    4.63  346.05   20.52  345.53   23.14  344.66   27.92  344.29
   30.32   344.4   30.98  342.83   31.83  342.23   34.82  342.09   36.74  341.58
   46.45   341.2   46.96  340.92   47.56  340.78   48.68  339.84   50.39  338.81
   51.14  338.52   53.27  338.49   57.25  338.61   58.58   340.2   61.37  340.58
   64.54  340.56   73.16  340.77   87.05  340.61   88.25   340.7   89.02  341.37
   91.32  341.91   98.87  341.88  103.09  341.66   127.6  341.57  150.84  341.95
#Mann= 3 , 0 , 0
       0      .1       0   46.45     .04       0   61.37     .08       0
Levee=0,,,-1,60.53,341.9759,,	2160
#Block Obstruct= 5 ,-1
   20.56    21.8348.3146  111.76  126.89  344.59   73.17    84.9   343.7
       0    3.93349.2465  147.77  150.84344.9349
Bank Sta=46.45,61.37
XS Rating Curve= 0 ,0
Exp/Cntr=0.3,0.1

Type RM Length L Ch R = 1 ,15967.45,9.35,9.53,9.59
XS GIS Cut Line= 5
-610992.09319999   -1045900.0587    -611013.8884   -1045860.6581
-611022.15659999   -1045848.0903-611039.60269999   -1045797.2262
-611042.06069999   -1045753.1775
#Sta/Elev= 26
       0  347.27   17.76  346.49   26.01  341.96   28.84  341.41   33.02   341.2
   37.08  341.42   43.15  341.23   45.64  341.05   46.95  339.37    47.7  338.52
   51.85  338.33   55.01  338.41   55.61  339.89   56.02  340.12   56.35  340.16
   61.82  340.34   62.73  340.49    75.1  340.45   83.56  340.67   89.14  340.62
    90.5   340.7   92.58  341.68  109.06  340.95   125.8  341.47  141.22  341.59
  157.96  341.87
#Mann= 3 , 0 , 0
       0      .1       0   45.64     .04       0   56.35     .08       0
Levee=0,,,-1,57.76,341.7307,,	2160
#Block Obstruct= 3 ,-1
  110.54  122.37344.1635       0    5.65350.1486  152.96  157.96344.8275
Bank Sta=45.64,56.35
XS Rating Curve= 0 ,0
Exp/Cntr=0.3,0.1

Type RM Length L Ch R = 1 ,15957.93,15.71,14.65,13.63
XS GIS Cut Line= 5
     -611000.734   -1045904.2531    -611020.2591   -1045868.1678
-611030.47859999   -1045852.8987-611045.06769999   -1045811.8192
-611048.78449999   -1045753.7894
#Sta/Elev= 30
       0  347.88    4.05   347.4   15.74  346.67   21.67   342.3   22.34  342.03
   36.42  341.29    43.5  341.24   43.53  341.44   43.83  341.45   43.88  340.76
   44.08  340.53   44.92  340.42   44.94  340.49   44.95  338.61   50.61  338.18
   53.89  338.28    54.2  339.05   54.58   339.2   55.32  340.08   62.03  340.33
   77.96  340.18   85.16  340.35   91.04  340.72   92.73  341.52  114.67  340.85
  124.49  341.18  129.49  341.21  136.74  341.55   144.9  341.61  161.14  341.96
#Mann= 3 , 0 , 0
       0      .1       0   43.83     .04       0   55.32     .08       0
Levee=0,,,-1,55.65,341.5947,,	2160
#Block Obstruct= 4 ,-1
  118.77  121.07344.0259  101.15   106.8344.1338       0    4.09350.6369
   28.65   36.42344.4799
Bank Sta=43.83,55.32
XS Rating Curve= 0 ,0
Exp/Cntr=0.3,0.1

Type RM Length L Ch R = 1 ,15943.28,9.23,8.7,8.01
XS GIS Cut Line= 5
-611018.45259999   -1045911.2168    -611035.5181   -1045872.8951
-611044.51399999   -1045854.9034-611060.44139999   -1045803.4049
-611062.47329999   -1045751.5215
#Sta/Elev= 30
       0  346.99   11.75  346.51   15.23  343.43   16.49  342.17    18.6  341.78
   20.91  341.53   23.32   341.1   36.13  341.38   43.42  341.31   43.45  341.42
   43.94  341.41   43.98  338.67   43.99  338.44   47.44  338.01    50.9  338.25
   51.56  338.86   53.14  339.97    70.6  340.34   70.79  340.21   77.82   340.1
   80.64  340.16   86.13  340.43   89.75  340.75   90.69  340.92   91.59  341.39
  120.67  340.85  140.07  341.08  148.45  341.48  156.33  341.58  167.89  341.86
#Mann= 3 , 0 , 0
       0      .1       0   43.94     .04       0   53.14     .08       0
Levee=0,,,-1,53.22,341.4764,,	2160
#Block Obstruct= 4 ,-1
       0    5.87349.8845    69.9   77.54 343.214   80.86   87.63 343.366
     100  110.29344.1213
Bank Sta=43.94,53.14
XS Rating Curve= 0 ,0
Exp/Cntr=0.3,0.1

Type RM Length L Ch R = 1 ,15916.88,28.68,28.89,29.62
XS GIS Cut Line= 5
    -611049.8937   -1045915.0428    -611060.9182    -1045881.891
    -611064.3608   -1045872.7106    -611083.0196   -1045801.8009
-611091.84849999   -1045749.5303
#Sta/Elev= 30
       0  346.99     .14  346.97    1.35  346.23    3.51   344.3    7.42  344.34
    11.8  344.15   14.85  342.27   27.72  341.29    36.4  340.97   37.45  341.06
   37.46  339.45   37.49  337.94   40.08  337.77   43.05  338.06   45.05  339.83
   50.76     340   59.07  339.79   69.07  339.79   69.08  341.04   73.71  340.94
   74.31   340.2   91.65  341.44   93.35  340.37  101.08   340.6   101.5  340.85
  101.99   340.7   135.2   341.3  147.48  341.31  160.85  341.59  171.08   341.6
#Mann= 3 , 0 , 0
       0      .1       0   37.45     .04       0   45.05     .08       0
Levee=0,,,-1,44.99,341.2633,,	2160
#Block Obstruct= 2 ,-1
   54.77   62.06342.8527   14.11    27.7 345.008
Bank Sta=37.45,45.05
XS Rating Curve= 0 ,0
Exp/Cntr=0.3,0.1

Type RM Length L Ch R = 1 ,15829.9 ,19.46,19.19,18.61
XS GIS Cut Line= 4
-611127.02369999   -1045962.5109-611145.18809999   -1045901.2055
    -611151.8026   -1045882.0232    -611169.1645    -1045742.966
#Sta/Elev= 28
       0  345.48   10.89  346.08   13.33  346.15   19.07  345.57   22.36   343.9
    25.6  341.69   28.57  341.53   36.77  340.51   57.75  340.26   58.86  340.35
   67.39  339.84    67.4  337.35   76.27  337.37   76.28  339.16   76.36  339.17
   90.51  339.98   96.45  340.17  106.54  340.23  117.37  339.88  121.19  339.61
  137.99   340.9  151.71  341.32  181.95  341.29  186.38  341.17  197.12  341.09
  212.17  341.14   218.2  341.05  224.37  341.08
#Mann= 3 , 0 , 0
       0      .1       0   67.39    .035       0   76.36     .08       0
#Block Obstruct= 3 ,-1
   37.64   50.42343.4244  123.19  130.76343.0505  181.09   189.9344.2119
Bank Sta=67.39,76.36
XS Rating Curve= 0 ,0
Exp/Cntr=0.3,0.1

Type RM Length L Ch R = 1 ,15810.7 ,23.98,23.78,23.78
XS GIS Cut Line= 4
-611147.12029999   -1045960.8525-611163.70899999   -1045907.1587
-611169.66209999   -1045887.9764    -611188.3553   -1045742.9866
#Sta/Elev= 29
       0  345.46    6.47  345.37   10.74  343.06   11.78  342.35   13.26  341.49
   16.26  341.38   17.47  341.17   24.31  340.93   29.01  340.19    41.3  340.12
   43.17  340.04   57.56  340.02   60.31  337.52   60.32  337.35   68.62  337.49
   68.63  339.39   71.01  339.18   72.44  339.17   72.96     339   89.18  339.66
    92.7  339.69  104.49  340.31  119.55  340.35  149.92  340.86   172.8  341.05
   180.1  341.04  186.59  340.86  194.88  340.88  222.47  341.17
#Mann= 3 , 0 , 0
       0      .1       0   57.56     .04       0   68.63     .08       0
Levee=0,,,-1,69.14,339.23,,
#Block Obstruct= 1 ,-1
   191.2  211.22343.9536
Bank Sta=57.56,68.63
XS Rating Curve= 0 ,0
Exp/Cntr=0.3,0.1

Type RM Length L Ch R = 1 ,15786.92,22.11,20.36,18.99
XS GIS Cut Line= 4
     -611165.032   -1045987.8568    -611187.5216   -1045911.1275
-611192.15179999    -1045894.591    -611251.6831   -1045628.0227
#Sta/Elev= 27
       0  345.36    8.56  345.43   19.87   345.4   22.95  345.28   25.17  344.47
   29.12  342.87   33.82   340.6   39.46  340.31   54.42  340.24   61.97  339.98
   81.93  339.84   81.94  337.46   90.61  337.48   90.62  339.36   99.95  338.39
  106.03  338.63  125.74  340.02  178.62  340.35  194.02  340.33  237.09  340.58
  250.73  340.58  260.41  340.42  274.87   340.4  325.38  340.72  332.41   340.7
  363.26  340.99  370.26  341.42
#Mann= 3 , 0 , 0
       0      .1       0   81.93    .035       0   90.62     .08       0
Levee=0,,,-1,90.99,339.3,,
#Block Obstruct= 8 ,-1
   56.21    66.3343.0709  221.93  229.93343.4889  329.69  336.18343.7225
  312.31  324.45343.6595     299  303.61343.5717       0     .15348.3615
  178.74  183.69343.3546  204.71  211.66343.3929
Bank Sta=81.93,90.62
XS Rating Curve= 0 ,0
Exp/Cntr=0.3,0.1

Type RM Length L Ch R = 1 ,15754.75,11.28,11.29,11.04
XS GIS Cut Line= 6
     -611230.918   -1045995.6999    -611231.2355   -1045970.9348
    -611221.0212    -1045885.914    -611257.3088   -1045780.7867
    -611261.6351    -1045742.032    -611258.0872   -1045598.3207
#Sta/Elev= 30
       0  344.87   28.12  343.58   33.36  341.38   45.38  340.31    62.5  339.97
    79.6   339.9   82.07  340.05   84.19  339.85   84.22  338.74   84.29  337.54
    84.3  337.05   93.74  337.88   93.75  337.89   93.83  339.24   94.91  339.25
   96.15  339.68   96.21  340.01  108.01  339.48  115.21  339.44  208.71  340.26
  253.27  340.34  257.54  340.13  268.64  340.01  269.15  340.38  275.01  340.42
   275.6  340.29  355.89  341.29  359.79  341.58  379.77  342.25  404.72  343.65
#Mann= 3 , 0 , 0
       0      .1       0   82.07    .035       0   96.21     .08       0
#Block Obstruct= 1 ,-1
    8.14   22.52347.1254
Bank Sta=82.07,96.21
XS Rating Curve= 0 ,0
Exp/Cntr=0.3,0.1

Type RM Length L Ch R = 1 ,15743.46,14.98,13.54,10.62
XS GIS Cut Line= 6
    -611270.7595   -1046004.5644    -611232.9684    -1045916.367
-611231.32099999   -1045898.0854-611268.45829999   -1045778.8404
    -611272.7846   -1045740.0857    -611269.2368   -1045596.3744
#Sta/Elev= 30
       0  344.12   25.61  341.99   41.43  340.09   49.41  339.68    56.6  339.48
   70.68  340.13   78.41  339.37   90.78  339.37  101.39  339.84  101.42  339.84
  101.43  337.14  111.14  338.01  111.23  338.95  112.36   339.1  113.11  339.54
  116.83  339.65  153.54  339.13  175.09  340.05  221.29  339.97  224.48  339.66
  233.43  340.29  272.77  340.03  310.69  340.47  327.95  339.96  347.21  340.05
  352.21   340.5  361.08   340.4  379.62  340.97  417.22  343.25  422.69     344
#Mann= 3 , 0 , 0
       0      .1       0  101.39    .035       0  112.36     .08       0
#Block Obstruct= 6 ,-1
       0    1.87347.0369   60.66   71.88342.8853   137.3  139.05342.1466
  214.83  218.71342.9147  259.38  272.25 343.048  308.26  312.29343.4149
Bank Sta=101.39,112.36
XS Rating Curve= 0 ,0
Exp/Cntr=0.3,0.1

Type RM Length L Ch R = 1 ,15729.91,23.06,22.01,19.38
XS GIS Cut Line= 6
    -611281.7885   -1046000.8759-611247.89779999   -1045913.8258
    -611243.0385   -1045896.2879    -611241.4543   -1045878.3214
    -611273.2296   -1045770.2109    -611285.8491   -1045607.2642
#Sta/Elev= 30
       0   344.2    5.36  343.93   10.38  341.41   12.22   340.8   34.88  340.79
    34.9  339.36   40.38  339.15    86.3  338.91   97.84  339.94   97.85  337.19
  107.83  337.99  107.89  338.03  107.94  338.63  109.25  338.95  112.92  339.18
  113.68  339.48  124.63  339.37  136.84  338.67  148.48  338.73  164.67  339.97
  212.71  339.75  226.96   340.2  236.88  339.96   300.3   340.2  317.72  339.79
  346.77  339.76  377.88  340.49   383.6  341.02  387.37  342.52  405.77  343.91
#Mann= 3 , 0 , 0
       0      .1       0   97.84    .035       0  109.25     .08       0
#Block Obstruct= 9 ,-1
  125.59  136.26342.0143  142.44  166.88342.3365     191  212.02 342.868
   56.85   77.08342.0844  300.27  334.05343.0232  253.06  265.89343.0455
  353.72  374.44343.1166  170.09  181.11342.9549   234.7  245.66343.0414
Bank Sta=97.84,109.25
XS Rating Curve= 0 ,0
Exp/Cntr=0.3,0.1

Type RM Length L Ch R = 1 ,15707.91,3.89,3.89,3.9
XS GIS Cut Line= 6
    -611297.0154   -1045997.0692-611269.98739999   -1045907.1252
    -611262.9829    -1045890.143    -611257.7215   -1045872.5269
    -611281.2811   -1045780.8493    -611297.0154   -1045616.4002
#Sta/Elev= 30
       0  346.46     .29  346.47     7.4  342.56   11.53  340.63   31.45  340.72
   31.46  339.07   57.35  339.29   68.02  338.94   95.25  338.87   97.93  339.43
   98.03  337.07   101.3  337.03  107.88  337.16  107.95  338.03  108.02  338.39
  115.25  338.84  130.67   338.9  143.77  338.47  159.13  339.67  174.73  339.56
  190.03  339.85  221.21  339.84  238.26  340.07  316.29  339.76  333.17  339.53
  357.76  340.21  371.62  340.94  372.23  340.76  386.69  343.84  390.53   344.3
#Mann= 3 , 0 , 0
       0      .1       0   97.93    .035       0  108.02     .08       0
#Block Obstruct= 6 ,-1
   39.03   57.74342.1694  291.09  330.12342.7108  195.81   209.7342.8094
  151.82  178.41342.3976  137.81  146.51341.7051  230.44  238.06343.0097
Bank Sta=97.93,108.02
XS Rating Curve= 0 ,0
Exp/Cntr=0.3,0.1

--- PPO_Kvasiny_efektiv.g02 (geometry) ---

Geom Title=N-Q10
Program Version=5.03

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
River Reach=Bela            ,Bela_reach

Type RM Length L Ch R = 1 ,19010.09,63.81,66.01,58.86
XS GIS Cut Line= 5
-608502.66209999   -1044593.6857    -608536.6251   -1044560.8986
     -608549.118   -1044545.2805    -608586.5786   -1044508.0775
     -608607.896   -1044465.4426
#Sta/Elev= 28
       0  393.68    6.75  390.81   16.83  386.16    26.9  380.59   29.66  378.85
   36.98  374.49   39.39  373.14   43.16  371.22   52.73  369.09   53.15 368.985
   53.94  367.04   60.45  367.16   64.36  370.18    64.4370.1805   70.18  370.38
   89.09  370.33   110.6  370.01  112.68  370.04     120  369.94  120.58  369.94
  122.07  369.15  134.59  369.48  137.58  369.42  142.28  370.49  146.47  372.64
  150.45  374.01  164.12  378.96  167.67  380.13
#Mann= 5 ,-1 , 0
       0     .15       0   53.15     .05       0    64.4      .1       0
  112.68     .05       0     120     .12       0
Bank Sta=52.73,64.36
XS Rating Curve= 0 ,0
Exp/Cntr=0.3,0.1

Type RM Length L Ch R = 1 ,18944.07,107.06,100,81.52
XS GIS Cut Line= 5
    -608546.4782   -1044642.7763-608578.86259999   -1044608.0005
     -608594.864   -1044596.0024    -608642.9144   -1044514.1948
    -608653.0656   -1044483.0645
#Sta/Elev= 29
       0  386.63   16.09  379.43   25.66  375.39   35.22  371.96   38.92  370.86
   44.79  369.39   48.23  369.42    49.8  369.23   51.56368.1339   54.36  366.39
   60.63  366.88   67.02  370.14   67.03370.1393   79.71  369.64   80.76  369.77
   83.72  369.44   97.93  368.72  116.15  369.27  118.16  369.71   127.9369.1595
  130.38  369.03  150.14  368.77  154.47   368.8  156.24  368.69  164.17  368.54
  165.15   369.7  173.57   373.4  187.32  378.52  195.14  382.34
#Mann= 5 ,-1 , 0
       0     .15       0   51.56     .05       0   67.03      .1       0
  118.16     .05       0   127.9     .15       0
#Block Obstruct= 1 ,-1
  137.23  152.56371.8682
Bank Sta=49.8,67.02
XS Rating Curve= 0 ,0
Exp/Cntr=0.3,0.1

Type RM Length L Ch R = 1 ,18844.07,72.16,72,73.34
XS GIS Cut Line= 6
-608649.34349999   -1044712.1427    -608661.1943   -1044671.2681
    -608666.6842   -1044652.0363-608687.57959999     -1044587.96
    -608711.2657   -1044551.4157    -608740.0273   -1044528.7448
#Sta/Elev= 28
       0  384.04   18.89  375.24   26.18  371.94   33.47  369.13    35.9   368.6
   40.75  367.36   44.03  368.88   44.31  369.11   44.35  369.09   44.67  368.93
   48.88  366.03   56.14   365.9   58.65  367.74   59.34  368.14   59.46368.1367
   70.03  367.79  101.43  368.09     118  368.06  120.69  368.11  122.41  368.58
  133.48  368.52  153.46  368.37  167.81  367.98  174.98   367.9  184.29  372.41
  191.95  376.82  197.36  379.79  210.13  386.07
#Mann= 5 ,-1 , 0
       0     .15       0   44.35     .05       0   59.46      .1       0
  122.41     .05       0  133.48      .1       0
Levee=-1,44.3,369.1,-1,59.9,368.04,,
Bank Sta=44.31,59.34
XS Rating Curve= 0 ,0
Exp/Cntr=0.3,0.1

Type RM Length L Ch R = 1 ,18772.07,49.5,53.87,46.34
XS GIS Cut Line= 5
-608717.01799999   -1044739.5508    -608729.3973    -1044693.413
    -608735.3242   -1044674.3114    -608762.3599   -1044598.1112
    -608783.6774   -1044558.5216
#Sta/Elev= 28
       0  383.29   18.17  376.48   32.67  370.79   39.91  368.37   47.16  366.81
   50.67  367.88   50.91  368.11   50.99368.0506   53.81  365.91    61.6  365.94
    64.7367.9844   64.71  367.99   66.95  367.36   69.23  367.23  114.85  367.42
     125  367.34  125.72  367.28   127.5  367.71  138.51  367.52  140.12  366.69
  141.02  367.28  148.38  366.93  149.49  366.52  154.63  369.91  178.71  385.11
  185.36  389.12  189.15  389.84  193.59  390.51
#Mann= 5 ,-1 , 0
       0     .15       0   50.99     .05       0    64.7      .1       0
   127.5     .05       0  138.51     .12       0
Levee=-1,50.87,368.11,-1,64.69,367.98,,
Bank Sta=50.91,64.71
XS Rating Curve= 0 ,0
Exp/Cntr=0.3,0.1

Type RM Length L Ch R = 1 ,18718.21,29.06,21.79,6.52
XS GIS Cut Line= 5
-608753.54699999   -1044753.4637     -608781.487   -1044705.5211
    -608789.4245   -1044670.2786    -608798.9496    -1044622.336
-608821.80959999   -1044578.8384
#Sta/Elev= 30
       0  384.35    4.01  382.93   12.11  379.51   16.79  376.59   28.31  368.13
   30.69  367.22   36.42  365.83   38.32  367.98   41.56  368.77   42.02  369.93
   45.86   364.9   46.37  364.88   51.77  364.89   54.68  367.03   71.29  366.92
    76.2  367.22   83.37  367.48   86.48  367.28   90.94  367.38  100.86  367.34
  117.53  367.08  134.11  367.25  140.49  367.21  143.13   367.2  144.27  366.52
  144.99  366.93  148.71  367.15  149.91  366.25  182.91  387.38  189.63   388.8
#Mann= 5 ,-1 , 0
       0     .12       0   42.02     .05       0   54.68     .05       0
  140.49     .05       0  149.91     .12       0
Levee=-1,42.02,369.93,-1,142.96,367.15,,
Bank Sta=42.02,54.68
XS Rating Curve= 0 ,0
Exp/Cntr=0.3,0.1
