HEC-RAS study PPO_Kvasiny_efektiv.prj: PPO_Kvasiny_efektivita

--- PPO_Kvasiny_efektiv.g02 (geometry) --- (continued)

Type RM Length L Ch R = 1 ,18696.42,50.22,38.35,4.09
XS GIS Cut Line= 4
-608796.05849999    -1044760.252    -608795.7939   -1044693.8414
    -608803.2023   -1044622.1392    -608824.1044   -1044584.3037
#Sta/Elev= 30
       0  380.28    3.25  378.85    9.27  375.53   16.25  371.11   17.25  370.36
   24.25  367.12   28.85   369.8   33.19     365   38.76  364.81   42.24  366.59
    42.5  366.59   46.19  366.81   53.31  366.69   70.21  366.94   78.14  367.19
   81.39  368.09   84.36  369.75   87.08  369.78   89.29     370   89.92  369.72
   93.55   367.5  115.58  366.97  130.78  367.24  139.61  367.19  140.83  366.48
  141.43  366.87  144.32  367.13  145.62  366.34   178.3  387.23  181.72  387.95
#Mann= 5 ,-1 , 0
       0      .2       0   28.85     .05       0    42.5     .15       0
  130.78     .05       0  140.83     .15       0
Levee=0,,,-1,87.99,369.73,,
#Block Obstruct= 1 ,-1
   99.66  107.48370.2419
Bank Sta=28.85,42.5
XS Rating Curve= 0 ,0
Exp/Cntr=0.3,0.1

Type RM Length L Ch R = 1 ,18658.06,22,33.51,26.87
XS GIS Cut Line= 6
-608811.08549999    -1044755.116     -608825.589   -1044701.0257
    -608807.8792   -1044691.7325-608803.30299999   -1044664.7705
    -608806.6867   -1044622.1356-608834.09479999   -1044582.8844
#Sta/Elev= 30
       0  378.22   12.72  374.61   27.41  371.22   36.15  368.78    43.1  367.32
    46.5  365.69   53.84  365.69   56.09  365.96   61.11  366.23   62.71   366.9
   62.73  364.21   69.51  364.09   70.75  365.09   74.45  366.52   74.46366.5206
   77.86  366.86   92.64  366.97   96.45  367.35  103.66  367.39  122.92   366.9
  134.34  367.11   142.8367.2064  146.19  367.18  147.55  366.45  148.03  366.83
  150.17  367.09  151.31  366.42  171.67  379.13  183.96  386.99  194.08  389.02
#Mann= 5 ,-1 , 0
       0      .2       0   62.71    .045       0   74.46     .12       0
  134.34     .05       0   142.8     .12       0
Levee=-1,62.62,366.83,-1,77.85,366.86,,
#Block Obstruct= 1 ,-1
  104.88  123.34370.1295
Bank Sta=62.71,74.45
XS Rating Curve= 0 ,0
Exp/Cntr=0.3,0.1

Type RM Length L Ch R = 1 ,18624.55,27.54,38.49,47.2
XS GIS Cut Line= 6
    -608813.3292   -1044757.0751-608830.65819999   -1044713.3605
     -608838.708   -1044671.6675    -608829.9133   -1044663.7088
    -608830.5483   -1044653.6758    -608851.3869   -1044598.6741
#Sta/Elev= 30
       0  378.92   15.14  374.94   22.67  373.16    30.2  371.61   40.84  368.61
   44.87  368.72   44.88  367.19   46.46  365.77   56.35  365.59   58.15  365.81
   71.85  365.45   85.93  366.54   89.66  367.02   89.67  364.06   98.15  364.03
   101.2  367.01  101.96   366.9  120.26  367.04  122.19  365.97  123.18  366.43
  124.31  367.04  129.18  367.16  132.12  367.14  133.58  366.63  136.31  368.67
  144.85  374.62  152.76  379.57  161.81  385.47  167.38  386.49  170.22  387.15
#Mann= 5 ,-1 , 0
       0      .2       0   89.66     .05       0   101.2     .12       0
  123.18     .05       0  133.58     .15       0
Levee=-1,88.65,366.51,0,,,,
#Block Obstruct= 2 ,-1
   43.76   47.02 370.226   55.44   78.67368.7872
Bank Sta=89.66,101.2
XS Rating Curve= 0 ,0
Exp/Cntr=0.3,0.1

Type RM Length L Ch R = 1 ,18533.27,12.87,12.37,12.43
XS GIS Cut Line= 4
    -608836.7278   -1044771.9928-608886.99879999   -1044726.4844
    -608909.2238   -1044709.0218    -608949.4406   -1044673.5676
#Sta/Elev= 29
       0   380.4   11.91  376.17   15.57  375.08   21.75  372.96   27.09  371.58
   30.64   370.1   34.92  368.53   43.78   368.6   45.25  367.34   53.98  366.18
   55.12  365.56   77.94  365.47   81.16  367.64   81.17  363.27   82.75  363.28
   90.22     363    91.2  363.02   92.37  365.49   92.53   365.6   93.52  365.72
   99.07   365.6   99.74   365.6   110.1  371.67  120.92  378.85  137.46  380.17
  138.48  380.28  141.03  380.97  141.59  381.06  149.69   381.6
#Mann= 4 ,-1 , 0
       0      .2       0   81.16    .035       0   92.53     .05       0
   99.07      .2       0
#Block Obstruct= 1 ,-1
   42.53   68.26370.0591
Bank Sta=81.16,92.53
XS Rating Curve= 0 ,0
Exp/Cntr=0.3,0.1

Type RM Length L Ch R = 1 ,18520.9 ,21.89,22.29,22.52
XS GIS Cut Line= 4
    -608863.4842   -1044765.4406-608906.08109999   -1044727.1808
-608921.42689999     -1044715.01    -608957.6926   -1044685.3842
#Sta/Elev= 27
       0  373.03    1.54  372.55   12.66  368.43   20.28  368.59   24.23  365.57
   42.35  365.58   53.42  365.42   54.89   366.7   56.03  367.47   56.04  362.99
   63.28  363.07   63.48   363.2   63.73  363.25   63.82  363.44   66.43  365.21
   67.69  365.49   73.85   365.4   76.67  367.07   77.16  367.22   80.37   368.9
    86.5  372.56   94.37  377.38  111.84  379.09  113.26  379.54  115.53  379.54
  118.39  380.28  123.67  380.54
#Mann= 4 ,-1 , 0
       0      .2       0   56.03     .04       0   67.69     .05       0
   73.85      .2       0
#Block Obstruct= 1 ,-1
   30.89   43.04368.5746
Bank Sta=56.03,67.69
XS Rating Curve= 0 ,0
Exp/Cntr=0.3,0.1

Type RM Length L Ch R = 1 ,18498.6 ,2.83,3.09,3.31
XS GIS Cut Line= 4
    -608885.6669   -1044772.6373    -608919.2351   -1044745.1325
    -608935.1101   -1044732.9616    -608964.8046   -1044708.0749
#Sta/Elev= 29
       0  370.37    7.01  368.43   13.26  368.15   15.38  365.51   18.15  365.54
   28.73   365.4   31.54  365.25   35.05  365.41   43.04   365.6   43.11  365.66
   43.12  362.62   46.14  362.62   48.74  362.73   52.41  365.03   53.99  365.11
    59.4  365.05   67.77  370.02   69.23  370.47   72.79  372.34   73.35  372.39
   79.86  375.88   81.41  376.09    89.3  376.67   92.41  376.98   93.25  377.63
   93.77  377.75   99.93  377.81  100.78  377.34  102.15  377.32
#Mann= 4 ,-1 , 0
       0      .2       0   43.11     .04       0   52.41     .05       0
    59.4      .2       0
Bank Sta=43.11,52.41
XS Rating Curve= 0 ,0
Exp/Cntr=0.3,0.1

Type RM Length L Ch R = 1 ,18495.51,25.6,24.88,23.57
XS GIS Cut Line= 4
    -608887.9529   -1044774.1613    -608917.6792   -1044750.0879
    -608934.0835    -1044737.917    -608970.0669   -1044707.7544
#Sta/Elev= 27
       0  370.29    6.96  368.39   10.03  368.32   13.09  368.15   15.21  365.51
   21.57  365.46   28.43  365.09   37.14  365.48   42.19  365.61   44.14   362.6
   47.66  362.74   49.82   364.1   51.54  364.96   53.01  365.07   58.45     365
   67.51  370.43    69.1  370.93    70.8  371.82   71.62   371.9   74.81   373.6
    79.7  375.88   86.45  376.34   91.06   376.8  100.25  377.07  101.89  377.02
  102.68  377.63  105.63  377.96
#Mann= 4 ,-1 , 0
       0      .2       0   42.19    .045       0   51.54     .05       0
   58.45      .2       0
Levee=0,,,-1,52.01,366.5074,,	2157
#Block Obstruct= 1 ,-1
   16.66   42.27367.0693
Bank Sta=42.19,51.54
XS Rating Curve= 0 ,0
Exp/Cntr=0.3,0.1

Type RM Length L Ch R = 1 ,18470.63,5.16,5.37,5.75
XS GIS Cut Line= 4
-608906.65179999   -1044793.0242    -608930.3372   -1044772.7807
-608945.32779999   -1044759.5411    -608983.9917   -1044723.9844
#Sta/Elev= 30
       0  371.32    4.35  370.26   12.24  369.28    14.4  369.57   17.14   368.8
   18.23  368.32   19.27  368.09   22.05  367.88   25.79  366.79   26.47  366.47
   32.99  365.07   37.38     365      39365.5917   39.08  365.61    39.1  362.44
   41.97  362.32    44.8  362.51   48.59  364.64   49.46  364.74   55.09  364.67
   55.62   364.6   57.27  365.52   61.13  368.88   61.66  369.46   63.49  369.91
    66.2  371.32   80.07   371.9   85.24  374.71   96.53   375.1  103.69  376.28
#Mann= 4 ,-1 , 0
       0      .2       0      39    .045       0   48.59     .05       0
   55.09      .2       0
Levee=0,,,-1,48.46,366.0615,,	2157
#Block Obstruct= 1 ,-1
   23.55   39.08 367.954
Bank Sta=39.08,48.59
XS Rating Curve= 0 ,0
Exp/Cntr=0.3,0.1

Type RM Length L Ch R = 1 ,18465.26,17.65,17.49,17.14
XS GIS Cut Line= 2
    -608910.5632   -1044796.3117    -608988.7089   -1044730.0063
#Sta/Elev= 28
       0  371.42   13.27  369.79   14.51  369.96   17.78  369.04   21.24   367.9
   29.02   365.7   31.41  365.18   31.74  365.04    38.2  364.12    38.4  362.34
   40.87  362.26   43.62   362.4    47.5  364.56   48.04  364.63   53.93   364.6
    55.3  364.89   55.55  365.01   57.04   366.3   59.46  368.95   60.65  369.04
   61.48  369.46   61.85  369.53    65.4  371.37   79.92  371.68   84.67   374.5
   96.34  374.66   98.15  374.96  102.48   375.9
#Mann= 4 ,-1 , 0
       0      .2       0    38.2     .05       0   48.04     .05       0
   53.93      .2       0
Levee=0,,,-1,47.29,365.9167,,	2157
Bank Sta=38.2,48.04
XS Rating Curve= 0 ,0
Exp/Cntr=0.3,0.1

Type RM Length L Ch R = 1 ,18447.77,15.66,15.93,16.64
XS GIS Cut Line= 4
-608918.60229999   -1044812.6923-608948.38219999   -1044787.3387
    -608962.1406   -1044775.1678    -609000.7698   -1044738.6552
#Sta/Elev= 30
       0  372.91    4.15  371.81     8.4  371.14   27.27  369.11   34.52  367.51
   38.21  364.55   42.26  364.03   42.29  363.69   42.46  362.26   45.32  362.08
   48.21   362.2   51.24  364.26   51.65  364.38   57.48  364.36   57.63  364.35
   62.76  367.26   64.08  367.82   66.39  367.95   67.64   368.2   70.61  370.19
   72.34  371.24   76.82  371.37   77.73   371.6   81.68  371.98   90.92  372.23
   90.94  374.32     102  374.46  104.88  375.09  108.48  375.51  110.63  375.63
#Mann= 4 ,-1 , 0
       0      .2       0   42.26     .05       0   51.65     .05       0
   57.48      .2       0
Levee=0,,,-1,51.03,365.5753,,	2157
#Block Obstruct= 1 ,-1
   82.53   97.95376.1941
Bank Sta=42.26,51.65
XS Rating Curve= 0 ,0
Exp/Cntr=0.3,0.1

Type RM Length L Ch R = 1 ,18431.84,14.94,15.01,15.06
XS GIS Cut Line= 4
-608926.42619999   -1044827.1558    -608957.9395   -1044799.6768
-608973.81459999   -1044786.9768    -609015.6187   -1044748.3474
#Sta/Elev= 30
       0   373.9    3.28  373.01   17.77  370.61    21.2  370.57   25.16   369.8
   36.17  368.09   38.42  367.23   41.35  364.87   45.17  363.98   45.26  363.94
   45.46  362.11   48.45  361.93   51.55  362.08   53.78  364.01   54.56  364.12
   60.23  364.07   60.48  364.06   64.62  367.06   69.71  367.56   76.92  371.42
   78.95  371.58   82.79   374.2   98.96  374.35  101.93  373.19  104.34  373.46
  105.32  373.41  105.89  374.06  106.87  374.01  109.27  374.28  119.06  374.86
#Mann= 4 ,-1 , 0
       0      .2       0   45.17     .05       0   54.56     .05       0
   60.23     .15       0
Levee=0,,,-1,53.56,365.304,,	2157
Bank Sta=45.17,54.56
XS Rating Curve= 0 ,0
Exp/Cntr=0.3,0.1

Type RM Length L Ch R = 1 ,18416.83,19.51,19.31,18.8
XS GIS Cut Line= 4
    -608933.7448   -1044840.0106    -608967.9937   -1044810.7893
-608985.98539999   -1044796.5017    -609023.5562   -1044764.7517
#Sta/Elev= 27
       0  374.51   15.08  370.39   22.91  370.54   25.64  370.51   28.28  369.99
   41.04  365.27   45.46  364.12   48.01  363.02   48.12  361.95    53.3  361.78
   55.49  363.73   56.19  363.86   62.29  363.82   63.37  364.02   64.02  364.06
   64.91  364.31   67.23  364.48   74.88  365.43   82.25  368.43   91.55   369.8
   99.91  370.77  104.42  372.58  111.02  373.18  112.87  373.22  113.53   373.1
   114.8  373.37  117.19   373.5
#Mann= 4 ,-1 , 0
       0      .2       0   45.46     .05       0   56.19     .05       0
   62.29     .15       0
Levee=0,,,-1,55.47,365.2081,,	2157
Bank Sta=45.46,56.19
XS Rating Curve= 0 ,0
Exp/Cntr=0.3,0.1

Type RM Length L Ch R = 1 ,18397.53,7.24,7.17,6.9
XS GIS Cut Line= 4
-608943.77299999   -1044858.6939-608978.04789999   -1044827.7227
    -608998.6854   -1044810.2602    -609033.0813   -1044782.2143
#Sta/Elev= 29
       0  375.54   15.13  371.42   21.18   369.7   28.37  367.14   37.48  364.36
   37.74   364.2   38.84  364.19   42.41  363.74   49.36  363.54   50.95  362.46
   51.38  361.93   53.74  361.63   56.63  361.76   57.34  362.35   59.02  363.46
   59.91  363.63    65.7  363.51    67.3  363.03   68.82  364.02   74.78  364.59
   83.08  364.84   85.93  366.75   95.12  367.15   96.23  367.75   99.72  369.86
  103.29  370.38   113.2  371.23  116.84  371.32  117.61   371.4
#Mann= 4 ,-1 , 0
       0      .2       0   49.36     .05       0   59.91     .05       0
    65.7     .15       0
Levee=0,,,-1,58.91,364.8894,,	2157
Bank Sta=49.36,59.91
XS Rating Curve= 0 ,0
Exp/Cntr=0.3,0.1

Type RM Length L Ch R = 1 ,18390.36,15.99,15.59,15.07
XS GIS Cut Line= 2
    -608947.5425   -1044864.1187-609036.10399999   -1044786.5639
#Sta/Elev= 27
       0  375.74   22.38   369.5    35.5  364.73   36.92  364.29   37.32  364.05
   41.73  363.53    49.8  363.33   52.13  361.76   54.39  361.53   56.98  361.72
   59.42  363.37   59.95  363.54   65.19  363.43   66.02  363.41   67.81  362.92
   69.47  363.95   70.84  364.08   80.38  364.55   85.55  364.72   86.08  365.17
      87   366.2   87.62  366.13   93.87  366.31   98.34  368.77  106.14   369.9
  108.95  370.15  117.72  370.43
#Mann= 4 ,-1 , 0
       0      .2       0    49.8     .05       0   59.95     .05       0
   65.19     .15       0
Levee=0,,,-1,59.32,364.8086,,	2157
#Block Obstruct= 1 ,-1
   30.72   43.62368.0001
Bank Sta=49.8,59.95
XS Rating Curve= 0 ,0
Exp/Cntr=0.3,0.1

Type RM Length L Ch R = 1 ,18374.77,12.72,13.16,13.09
XS GIS Cut Line= 3
-608959.05689999   -1044877.1776-609013.50209999   -1044826.1352
-609048.81949999   -1044791.2347
#Sta/Elev= 30
       0   375.3   10.49  372.78      15  371.53   32.38  364.68   36.18   364.1
   41.76  363.61   43.91  363.54   45.61   363.3   50.25  363.18    50.4  363.05
   50.88  361.48   53.79  361.32   56.67  361.56   58.83  363.14   59.59  363.37
   65.56  363.23   69.04  363.48   69.57  363.77   75.91  364.14   82.26  364.21
   83.54  364.29   84.04  364.51   84.48  364.55    88.3  364.42   93.29  364.73
   99.22  366.73  104.13  367.35  112.15  368.12  118.98  368.43  124.28  369.54
#Mann= 4 ,-1 , 0
       0      .2       0   50.25     .05       0   59.59     .05       0
   65.56     .15       0
Levee=0,,,-1,59.01,364.6792,,	2157
#Block Obstruct= 2 ,-1
   30.77   43.17367.4476   43.17   45.61366.4337
Bank Sta=50.25,59.59
XS Rating Curve= 0 ,0
Exp/Cntr=0.3,0.1

Type RM Length L Ch R = 1 ,18361.61,12.22,11.56,10.47
XS GIS Cut Line= 3
    -608967.6932   -1044884.2694     -609015.221   -1044843.1214
-609052.62759999   -1044801.8585
#Sta/Elev= 30
       0  374.49   11.75  371.69   24.58  366.45   28.45  365.54   34.76  363.68
   39.38  362.95   47.67  363.21   50.08  361.39   52.34  361.26   54.92  361.49
   56.46  362.18   56.84   362.1    57.1  362.77    57.1  363.21   65.93  363.09
   66.18  362.54   66.26  363.08   66.97  363.08   66.97  362.55   68.93  363.26
   69.65  363.34   76.43  363.59   83.69  364.12   88.17  364.27   90.45  364.11
  101.29  364.51  107.11  365.44  112.43  365.73  117.17  366.78  118.56  367.67
#Mann= 4 ,-1 , 0
       0      .1       0   47.67     .05       0    57.1     .06       0
   65.93     .15       0
Levee=-1,46.84,363.17,-1,57.89,364.7152,,	2157
Bank Sta=47.67,57.1
XS Rating Curve= 0 ,0
Exp/Cntr=0.3,0.1

Type RM Length L Ch R = 1 ,18350.04,2,2,2.21
XS GIS Cut Line= 4
    -608978.2241   -1044895.2065    -609008.2817   -1044865.0536
-609022.72899999   -1044851.2234-609048.56549999   -1044818.2857
#Sta/Elev= 22
       0  373.57     9.6  371.52   13.82  370.74   28.98  366.75   29.65  366.55
    33.8  363.79   35.16  363.25   36.75   362.9   47.26  363.08    47.8  362.16
   49.92  361.34   52.39  361.21   55.19  361.41    56.2  361.99   57.62  363.12
   57.71  363.12   59.38  363.15    65.2     363    67.3  363.14   75.51  363.06
   96.41  364.13  104.44  364.33
#Mann= 4 ,-1 , 0
       0      .1       0   47.26     .05       0   57.71     .06       0
    67.3     .15       0
Levee=0,,,-1,58.38,364.6284,,	2157
Bank Sta=47.26,57.71
XS Rating Curve= 0 ,0
Exp/Cntr=0.5,0.3

Type RM Length L Ch R = 1 ,18348.04,7.11,6.87,7.11
XS GIS Cut Line= 4
    -608980.1664   -1044896.0904     -609009.671   -1044866.4922
-609024.11829999    -1044852.662-609051.48649999   -1044819.8097
#Sta/Elev= 23
       0   373.3    6.85  371.83   14.58  370.39   27.13  367.13   31.91  364.08
   32.82  363.72   33.93  363.69   37.54  362.88   47.11  363.08   47.12  362.22
    47.3  362.08   49.13  361.33   51.22  361.18   52.62  361.27   55.16  361.27
    56.9  362.79   58.56  363.11   64.54  362.98   66.68  363.12   71.95  363.09
   74.49  362.95   94.77  364.01  104.55  364.23
#Mann= 4 ,-1 , 0
       0      .1       0   47.11    .045       0   58.56     .07       0
   71.95     .15       0
Bank Sta=47.11,58.56
XS Rating Curve= 0 ,0
Exp/Cntr=0.5,0.3

Type RM Length L Ch R = 1 ,18341.17,3.64,3.82,3.48
XS GIS Cut Line= 3
    -608984.7855   -1044901.5539    -609031.6963   -1044854.4518
    -609056.4353   -1044826.8159
#Sta/Elev= 28
       0  372.94    2.13  372.61   20.54  369.17   21.45  368.93   21.89  368.65
   33.77  363.06   39.86  362.88   43.25  362.84   46.71  362.94   47.49  362.85
   49.56  361.32   51.05  361.09   52.02  361.21   52.09  361.14   52.43  361.14
    52.5  361.21   56.44  361.21    57.3  362.09   57.94  362.73   58.53  362.88
   59.63  363.03   65.57  362.92   66.48  362.98   67.49  363.04   74.34  362.62
   81.72  362.96   86.35  363.35  103.57  363.97
#Mann= 4 ,-1 , 0
       0      .1       0   47.49    .045       0    57.3     .07       0
   66.48     .15       0
Levee=0,,,-1,59.93,362.97,,
Bank Sta=47.49,58.53
XS Rating Curve= 0 ,0
Exp/Cntr=0.3,0.1

Type RM Length L Ch R = 1 ,18337.36,14.84,14.42,14.55
XS GIS Cut Line= 4
     -608988.397   -1044905.6744    -609016.6957   -1044874.6581
-609031.05539999   -1044860.7368-609065.50409999   -1044820.1635
#Sta/Elev= 28
       0  372.66    7.27  371.71   18.26  369.64   22.38  369.43   23.75  366.65
   32.89  362.99   44.01  362.82   47.08  362.88   47.98  362.78   49.83  361.33
   51.34  361.04    52.2  361.22   52.32   361.1   52.89   361.1      53  361.22
   57.05  361.22   57.45  361.63   58.55  362.73   59.06  362.85   60.24  362.98
   66.23  362.88   67.23  362.95   74.45  362.47   84.01  362.91   87.64  363.22
  100.82  363.72  111.88  364.06  115.21  364.08
#Mann= 4 ,-1 , 0
       0      .1       0   47.98    .045       0   57.45     .07       0
   67.23     .15       0
Levee=0,,,-1,60.21,362.99,,
#Block Obstruct= 1 ,-1
   28.28   43.46366.8377
Bank Sta=47.98,59.06
XS Rating Curve= 0 ,0
Exp/Cntr=0.3,0.1

Type RM Length L Ch R = 1 ,18322.93,16.56,16.4,16.08
XS GIS Cut Line= 2
    -608999.2052   -1044914.5843-609092.44469999   -1044816.5633
#Sta/Elev= 30
       0   371.6   11.32  370.72   17.22  369.69      22  369.71   26.56  363.14
   26.79  363.06   36.52  363.02    43.2  362.74   46.09  362.76   46.17362.5667
   46.35  362.41   46.64  362.44   48.34  361.15   50.46  361.14   50.66  360.94
   51.66  360.94   51.86  361.14   56.24361.1803   57.76  362.55   58.39  362.78
   65.92  362.78   67.09  362.35   68.75  362.34    85.2  362.75  103.25  363.53
   109.5  363.69  124.02  363.67  125.26  364.47   130.6   365.3  135.28  366.61
#Mann= 4 ,-1 , 0
       0      .1       0   46.17    .045       0   56.24     .07       0
   65.92     .15       0
Levee=0,,,-1,59.9,362.83,,
#Block Obstruct= 1 ,-1
   26.73   35.54366.0181
Bank Sta=46.09,58.39
XS Rating Curve= 0 ,0
Exp/Cntr=0.3,0.1

Type RM Length L Ch R = 1 ,18306.53,11.47,11.55,11.69
XS GIS Cut Line= 3
-609011.42359999   -1044926.7722     -609089.892   -1044841.4859
-609102.89469999   -1044819.0525
#Sta/Elev= 30
       0  371.18    6.19  370.79   12.56  370.67   15.64  369.97   21.26   369.1
   28.33  363.04    42.1  362.52   42.75  362.52   42.97  362.64   43.53  362.67
   46.24  362.61   46.81  362.48   48.71  360.95   51.35  360.95   51.55  360.75
   52.55  360.75   52.75  360.95   56.63  360.95   56.76361.0543   58.26  362.25
   59.68  362.77   67.32  362.66   68.74  361.99   85.01  362.37   97.26  363.06
  115.89  363.41  131.24  363.56  131.94  364.19  136.75  364.86  141.82  366.12
#Mann= 4 ,-1 , 0
       0      .1       0   46.81    .045       0   56.76     .07       0
   67.32     .15       0
Levee=0,,,-1,60.51,362.67,,
#Block Obstruct= 2 ,-1
   39.21   42.75365.5524   76.18   94.88 365.575
Bank Sta=46.24,59.68
XS Rating Curve= 0 ,0
Exp/Cntr=0.3,0.1

Type RM Length L Ch R = 1 ,18294.98,16.32,15.92,15.19
XS GIS Cut Line= 4
    -609019.4125   -1044934.5905    -609077.4164   -1044872.4435
    -609103.2397   -1044839.8467    -609108.1081   -1044820.1617
#Sta/Elev= 30
       0  370.98    4.19  370.91   17.42  370.05   20.37  369.57   23.32  368.91
   26.83  366.55   34.78   362.5    43.3  362.56   46.18  362.42   47.13  362.35
   47.22  362.11   48.94  360.81   51.43  360.81   51.63  360.61   52.63  360.61
   52.83  360.81   56.87  360.81   57.35  360.81   58.98  362.11   60.37  362.62
   68.21  362.57   69.87  361.74   81.35  362.14   90.37  362.32  106.65  363.15
  129.28  363.42  136.27  363.36  136.81  363.82  142.18  364.59  146.87  365.89
#Mann= 4 ,-1 , 0
       0      .1       0   47.13     .05       0   56.87     .07       0
   68.21     .15       0
Levee=0,,,-1,61.52,362.56,,
Bank Sta=46.18,60.37
XS Rating Curve= 0 ,0
Exp/Cntr=0.3,0.1

Type RM Length L Ch R = 1 ,18279.06,5.31,5.32,5.33
XS GIS Cut Line= 5
-609032.27279999   -1044946.5812    -609059.4153   -1044915.6818
     -609083.818   -1044887.4375-609116.26419999   -1044848.5425
-609124.47399999   -1044813.5362
#Sta/Elev= 30
       0  372.24     1.5  372.25   15.72  369.87   19.55  369.35   23.91  369.19
   26.11  368.71   29.13  368.34   32.56  365.49   35.93  362.09   43.99  362.42
   46.63  362.26   48.93  360.62   51.46  360.62   51.66  360.42   52.66  360.42
   52.86  360.62   56.73  360.62   58.03  360.62   59.66  361.92   61.01  362.41
   69.03  362.46   70.79   361.7   95.28  362.05  101.69  362.42  106.65  362.88
  137.65  363.14  143.62  362.91     144  363.26  151.97   364.2  165.06  367.28
#Mann= 4 ,-1 , 0
       0      .1       0   46.63    .045       0   56.73     .07       0
   69.03     .15       0
Levee=-1,43.75,362.38,-1,62.46,362.46,,
#Block Obstruct= 1 ,-1
    85.1  103.82365.3277
Bank Sta=46.63,61.01
XS Rating Curve= 0 ,0
Exp/Cntr=0.3,0.1

Type RM Length L Ch R = 1 ,18273.75,10.28,9.7,8.84
XS GIS Cut Line= 5
    -609036.4443   -1044949.8598-609064.65399999   -1044917.7456
-609089.05669999   -1044889.5013-609120.98169999   -1044852.9628
    -609132.1506   -1044815.9045
#Sta/Elev= 30
       0  371.64     5.2  371.19   16.67   369.3   21.28  367.85      29  367.62
   33.77  364.43   35.92  362.28   38.55  362.42   46.12  362.24   46.23  362.15
   48.93  360.18   51.39  360.18   51.59  359.98   52.59  359.98   52.79  360.18
   57.28  360.18   57.82 360.614    59.4  361.88   60.82  362.35    68.5  362.42
   68.85  362.41   70.63  361.65   94.71   362.2  104.69  362.78  125.75   363.1
  141.77  363.11  145.94  362.92  146.35  363.21  157.05   364.3   167.3  366.38
#Mann= 4 ,-1 , 0
       0      .1       0   46.23    .045       0   57.82     .07       0
    68.5     .15       0
Levee=0,,,-1,63.29,362.42,,
#Block Obstruct= 1 ,-1
   86.04  104.85365.4245
Bank Sta=46.12,60.82
XS Rating Curve= 0 ,0
Exp/Cntr=0.3,0.1

Type RM Length L Ch R = 1 ,18264.04,12.48,12.71,12.7
XS GIS Cut Line= 5
    -609043.6799   -1044956.0504    -609072.4114   -1044924.5346
-609084.51969999   -1044908.6165    -609125.8273   -1044857.4816
-609142.94559999   -1044817.4285
#Sta/Elev= 30
       0  370.31   12.28  369.16   15.21  368.69   17.39   367.5   25.74  366.82
    37.8  361.96   41.05  362.18   45.27  362.15   46.56  361.95   47.29  361.26
   47.47   360.3   53.13   360.2   57.68  360.44   58.07  361.27   59.09   362.2
   61.57  362.11   63.06  362.35   68.94  362.33   70.89  361.61    72.5  361.89
   88.18  361.87   88.96  362.28   90.18  362.38  112.24  362.77  146.92  363.09
  148.75  362.97  149.04  363.13  153.37  363.53  164.13  364.28  171.94  365.37
#Mann= 4 ,-1 , 0
       0      .1       0   45.27     .05       0   59.09     .07       0
   68.94     .15       0
Levee=0,,,-1,62.77,362.26,,
Bank Sta=45.27,59.09
XS Rating Curve= 0 ,0
Exp/Cntr=0.3,0.1

Type RM Length L Ch R = 1 ,18239.54,14.41,15.04,15.89
XS GIS Cut Line= 3
    -609064.9836   -1044971.8533    -609104.8405   -1044922.9878
-609156.10359999   -1044845.2663
#Sta/Elev= 22
       0  366.86   11.26  365.81   13.62  365.34   14.21  365.31   15.61  364.85
   27.82  362.48   34.65  362.18   44.59  362.01   47.05  360.16   56.76  360.29
   60.01  361.98   68.06  362.02   68.68  361.65   69.15  361.22   70.05  361.57
   78.08  361.61   80.15  361.51    87.7  361.56   89.14  362.21  114.25   362.8
  123.01  362.88  156.16  362.72
#Mann= 4 ,-1 , 0
       0      .1       0   44.59     .05       0   60.01     .07       0
   68.06     .15       0
Levee=0,,,-1,60.6,361.97,,
#Block Obstruct= 2 ,-1
   16.12   37.69366.4533  101.13  121.79365.6882
Bank Sta=44.59,60.01
XS Rating Curve= 0 ,0
Exp/Cntr=0.3,0.1

Type RM Length L Ch R = 1 ,18224.5 ,18.07,18.46,18.77
XS GIS Cut Line= 3
    -609075.6612   -1044979.0075    -609117.0775    -1044932.579
-609210.79199999   -1044805.8233
#Sta/Elev= 28
       0  365.11   10.49  364.17   13.68  363.68   26.24  362.67   41.24  362.03
   43.28     362   43.96  361.76   46.43  360.03   48.49  359.94    55.2  360.03
   57.34  361.78   66.26  361.87   67.31  360.99   68.09  361.51   70.76  361.49
   84.16  361.75   86.64  361.61    87.3  361.49      90  361.78   102.4  362.52
  108.88  362.59  158.83  362.54  177.06  362.44  196.05  362.67  204.95  363.03
  214.11  363.16  215.94  363.32  219.85  363.87
#Mann= 4 ,-1 , 0
       0      .1       0   43.28     .05       0   57.34     .07       0
   66.26      .2       0
Levee=0,,,-1,58.17,361.72,,
#Block Obstruct= 1 ,-1
   17.57   28.26365.9847
Bank Sta=43.28,57.34
XS Rating Curve= 0 ,0
Exp/Cntr=0.3,0.1

Type RM Length L Ch R = 1 ,18206.04,5.09,4.98,4.99
XS GIS Cut Line= 4
     -609080.951    -1044998.105    -609116.2027    -1044960.872
    -609129.9171   -1044946.3148-609272.49179999   -1044770.8857
#Sta/Elev= 30
       0  367.22    4.83  366.36    6.94  366.52    8.97  365.99   12.57   364.3
   14.78  363.49   28.27  362.63   55.41   362.2   55.65  361.65      56  359.96
    58.7  359.69   63.69  359.58   65.74  359.86   65.96  360.26   66.01  361.53
   66.11  361.55   66.12   361.7   68.84  361.82   77.27  361.64    78.3  360.92
   79.13  361.48   90.93  361.17  129.25   362.2  170.35  361.86     247  362.15
  252.55  362.43  264.74  363.43  279.08  365.99   280.2  366.37  297.33  368.69
#Mann= 4 ,-1 , 0
       0      .1       0   55.41     .05       0   66.12     .07       0
   77.27      .2       0
Levee=0,,,-1,69.11,361.76,,
Bank Sta=55.41,66.12
XS Rating Curve= 0 ,0
Exp/Cntr=0.5,0.3

Type RM Length L Ch R = 1 ,18201.06,23.86,23.02,22.09
XS GIS Cut Line= 4
     -609081.967   -1045006.5717-609120.09479999    -1044964.001
    -609133.8092   -1044949.4436    -609276.3839   -1044774.0146
#Sta/Elev= 30
       0  370.45     4.8  370.18    9.09  368.12   16.22  367.74   26.16  363.16
    34.1  362.62   38.88  362.59   49.59  362.04   61.21  362.12   61.43  361.72
   62.15  359.61   63.21   359.5   70.02  359.52   70.68  359.73   71.92  361.91
   83.07  361.59   84.04  360.91   84.84  361.47   94.82  361.15  102.39  361.66
  115.93  361.61  134.35  362.12  200.36  361.64   211.5   361.1  215.58  361.35
  219.39     362  259.37  362.04  269.05  363.42  272.69  363.62  303.21  368.19
#Mann= 4 ,-1 , 0
       0     .15       0   61.21     .05       0   71.92     .07       0
   83.07      .2       0
Levee=0,,,-1,73.15,361.83,,
#Block Obstruct= 1 ,-1
    3.93   17.13371.7588
Bank Sta=61.21,71.92
XS Rating Curve= 0 ,0
Exp/Cntr=0.5,0.3

Type RM Length L Ch R = 1 ,18178.04,32.9,33.23,33.2
XS GIS Cut Line= 4
    -609103.6508   -1045021.0811-609138.55079999   -1044978.8772
    -609151.1605   -1044963.3531    -609291.7859   -1044770.6855
#Sta/Elev= 30
       0  370.22    4.28  368.69   21.67  367.17   22.82  366.86   27.24  364.45
   32.28  364.28    34.4  363.32   47.53  361.85   54.36  361.67   56.22360.7247
   59.04  359.39   62.85  359.24   66.74  359.62   67.19  359.89   73.29 361.474
   73.82  361.58   80.03  361.53   80.86  360.85   81.81  361.33  116.27  361.85
  148.98  361.84   172.7  361.43   230.3  361.73  231.77  361.18  233.41  361.85
   264.6  361.63  270.94  361.97  275.13  361.92  301.82  367.24  313.29   368.9
#Mann= 3 ,-1 , 0
       0     .15       0   56.22     .05       0   73.29     .15       0
Levee=0,,,-1,73.96,361.53,,
#Block Obstruct= 1 ,-1
  115.17  115.55 364.834
Bank Sta=54.36,73.82
XS Rating Curve= 0 ,0
Exp/Cntr=0.3,0.1

Type RM Length L Ch R = 1 ,18144.81,57.17,57.54,57.11
XS GIS Cut Line= 3
    -609126.6578   -1045045.0457    -609180.4545    -1044979.726
-609309.43919999   -1044786.5799
#Sta/Elev= 30
       0   370.4     .58  370.52     2.5   370.3   12.98  368.64   31.96   367.1
   35.49  365.19   38.21  364.92   53.14  365.02   55.75  362.09   56.66  361.95
   59.82  359.11   62.82  359.45   63.07  358.48   66.88  358.93   68.42  360.71
   73.26  361.12   98.47  361.22  119.71  361.61  126.56  361.47  144.56  361.63
  191.84  361.19  218.85  361.47  255.53  361.29  256.86  360.96  258.24  361.47
  272.83  361.32  287.16  361.78  304.06   365.5   307.2  366.01  316.88  367.05
#Mann= 3 , 0 , 0
       0     .15       0   56.66     .05       0   73.26     .15       0
#Block Obstruct= 1 ,-1
   91.09   102.3364.2794
Bank Sta=56.66,73.26
XS Rating Curve= 0 ,0
Exp/Cntr=0.3,0.1

Type RM Length L Ch R = 1 ,18087.28,17.9,17.24,16.41
XS GIS Cut Line= 4
    -609172.6953   -1045075.7374-609210.22019999   -1045033.9658
    -609225.4338   -1045014.7835-609349.78819999   -1044815.6841
#Sta/Elev= 30
       0  369.87     .34  369.79     1.9  369.76    8.72  369.06   17.99  368.63
   26.56  367.86   33.53  365.61   38.32  364.54   43.62  364.42   49.35  364.17
   57.84  358.79   65.35  358.82   67.14  360.31   71.92  360.44   74.13   360.4
   79.88  360.64   92.26  360.97  108.58  361.05  136.13  361.02  152.81  360.89
   185.2  360.93  215.99   360.6  236.03  360.54   237.4  360.02  238.91  360.69
  272.48  360.49  286.86  361.18  292.07  361.55  306.19  363.28  315.38  364.18
#Mann= 3 , 0 , 0
       0     .15       0   49.35     .05       0   67.14     .15       0
#Block Obstruct= 2 ,-1
    1.34   26.94371.7567  171.18  179.93363.9105
Bank Sta=49.35,67.14
XS Rating Curve= 0 ,0
Exp/Cntr=0.3,0.1

Type RM Length L Ch R = 1 ,18044.69,39.68,37.85,34.98
XS GIS Cut Line= 4
    -609211.3246   -1045101.1375    -609241.9703   -1045063.7315
    -609258.5068   -1045037.9345    -609384.8456   -1044831.5591
#Sta/Elev= 30
       0  369.31    2.39  369.32   19.27  368.35   22.94  368.32   23.29  367.96
   25.53  366.85   30.81  366.28   34.45  366.19   44.62  364.96   48.36  361.71
   52.05  358.11   60.57  358.01   60.99  358.01      61  360.18   63.04  359.73
   89.32  360.45  107.65  360.45   114.4  360.28  170.26  360.44  187.43  360.13
  198.58  360.24  215.58  360.05  239.86  360.35  241.36  359.56  242.68  360.34
  258.25  360.37  270.11  359.83  275.91   360.3  293.32  360.54  320.97  362.15
#Mann= 3 , 0 , 0
       0     .15       0   48.36     .05       0      61     .15       0
Levee=0,,,-1,61.43,360.05,,
#Block Obstruct= 4 ,-1
   36.85   45.32 368.134   69.09   78.84363.0494  299.39  309.67364.1195
  320.66  320.97365.1357
Bank Sta=48.36,61
XS Rating Curve= 0 ,0
Exp/Cntr=0.3,0.1

Type RM Length L Ch R = 1 ,18006.85,47.57,48.82,45.88
XS GIS Cut Line= 4
-609249.95389999   -1045127.0667-609280.33489999   -1045075.6377
    -609281.6579   -1045067.0388    -609407.3352   -1044850.7415
#Sta/Elev= 30
       0  369.21    4.91  368.61   13.43  367.83   16.58   367.1    22.5   366.3
   23.75  365.83      25  365.57   29.46  365.28   31.22  364.65   38.82  361.11
   39.25  361.61   48.26  359.62   59.73   359.4   60.41  358.92   60.42  357.47
    66.7  357.73   67.07  358.39   68.43  359.57   82.73   359.3   94.22  359.68
  122.56  359.96  160.18  359.69  170.96   359.9  194.24  359.82  248.41  360.07
  258.94   360.3  279.72  360.32  296.07  360.58  308.35  360.93  318.59  361.45
#Mann= 3 , 0 , 0
       0     .15       0   59.73     .05       0   68.43     .15       0
Levee=0,,,-1,68.59,359.54,,
#Block Obstruct= 1 ,-1
   74.05    85.4362.3846
Bank Sta=59.73,68.43
XS Rating Curve= 0 ,0
Exp/Cntr=0.3,0.1

Type RM Length L Ch R = 1 ,17958.03,4.98,4.96,5.01
XS GIS Cut Line= 5
-609289.07889999   -1045149.6626    -609326.2672   -1045090.5068
    -609331.3531   -1045071.1643-609362.16739999   -1045001.6811
     -609463.228   -1044828.8855
#Sta/Elev= 30
       0  369.29   10.49  367.12   14.99  366.62   22.52  362.14   25.14  361.66
   48.53   359.5   60.23  359.41   60.84  358.54   61.76  359.58   70.13  359.78
   75.55 359.302    75.8   359.3   75.82  357.91   79.63  357.53    84.3  357.64
   84.42  358.13   85.85  358.13   85.91  359.33   86.02359.3391   88.33  359.73
  100.05  359.74  101.16  359.17  113.29  359.09  128.04  359.49  246.69  359.43
  300.86  359.83  339.45  361.39  344.75  362.14  352.79  362.59  366.06  364.66
#Mann= 3 ,-1 , 0
       0     .15       0   75.55     .04       0   86.02     .15       0
Levee=-1,70.67,359.7,-1,88.68,359.7,,
#Block Obstruct= 1 ,-1
   137.4   140.4362.4691
Bank Sta=75.55,86.02
XS Rating Curve= 0 ,0
Exp/Cntr=0.5,0.3

Type RM Length L Ch R = 1 ,17953.06,18.09,19.04,21.99
XS GIS Cut Line= 5
    -609293.7773   -1045151.3166    -609330.9657   -1045092.1607
    -609336.0515   -1045072.8183    -609366.8658   -1045003.3351
-609467.92639999   -1044830.5395
#Sta/Elev= 30
       0  369.07    11.2  366.99   16.25  366.54   23.81  361.64   31.67  361.21
   34.54  359.98   49.71  359.02   55.47  359.16   56.39  358.03   57.93  359.51
   75.67   359.3   75.68  357.75   75.77  357.73   83.46  357.58   84.45  357.61
   84.51  358.04   86.02  357.94   86.03  358.73   86.12  358.74   86.13  359.33
   88.09  359.64  117.88  359.15     130   359.5  300.62  359.77  332.39     361
  334.26  362.21  336.13  362.19  336.58  361.57  354.75  362.83  366.06  365.13
#Mann= 3 , 0 , 0
       0     .15       0   75.67     .04       0   86.13     .15       0
Levee=-1,66.05,359.48,-1,89.61,359.48,,
Bank Sta=75.67,86.13
XS Rating Curve= 0 ,0
Exp/Cntr=0.5,0.3

Type RM Length L Ch R = 1 ,17934.03,65.98,74.44,72.11
XS GIS Cut Line= 5
    -609319.7439   -1045164.6074-609346.21489999    -1045097.348
    -609356.5102   -1045080.2014-609385.44929999   -1045009.9555
    -609484.1037    -1044838.313
#Sta/Elev= 30
       0  369.98    4.24  370.22     6.8  369.31   10.23  368.96   10.42  368.14
    18.3  367.33   23.78   362.9   27.99   362.3   36.51  359.32   52.99   358.4
   54.67  357.65   57.58  359.02   76.56   358.8   78.51  357.62   84.98  357.26
   85.93  357.35   88.49  358.89   94.07  359.24  120.45  358.94  180.97   359.7
   185.5  359.25  295.12  359.45   312.5  360.15  328.34  360.25  331.09  361.19
  343.38  361.45  347.01  361.72  352.88  362.67   359.2  364.58  366.23  367.65
#Mann= 3 ,-1 , 0
       0     .15       0   76.56     .04       0    88.7     .15       0
Levee=-1,66.74,358.96,-1,94.23,359.25,,
Bank Sta=76.56,88.49
XS Rating Curve= 0 ,0
Exp/Cntr=0.3,0.1

Type RM Length L Ch R = 1 ,17857.16,23.71,17.14,11.38
XS GIS Cut Line= 6
    -609389.2674   -1045183.2983-609397.27959999   -1045146.3236
-609413.71029999   -1045137.2749    -609412.9959   -1045133.7824
-609422.20239999   -1045089.9074    -609542.6629   -1044860.2654
#Sta/Elev= 30
       0  371.05   11.88  370.04   21.73  370.07   27.19  366.39   33.34  365.48
   38.94  360.97   39.59  359.83   41.94   358.6   42.26  357.26   42.66  356.66
   42.95  355.25   48.54   355.2   56.92  355.33   57.37  358.08   58.25  357.99
   58.31  357.04   59.65  356.96   59.87  358.11  104.85   358.6   105.7  357.95
  106.21  358.68  294.39  358.65  306.56  359.53  324.74  361.89     334  365.85
   336.2  365.98  337.98   366.9  355.28   369.2  362.81  371.82   364.3  371.12
#Mann= 3 , 0 , 0
       0     .15       0   41.94     .05       0   57.37     .15       0
Levee=0,,,-1,57.79,358.05,,
#Block Obstruct= 1 ,-1
       0    2.05373.9771
Bank Sta=41.94,57.37
XS Rating Curve= 0 ,0
Exp/Cntr=0.3,0.1

Type RM Length L Ch R = 1 ,17840.02,57.92,57.13,54.77
XS GIS Cut Line= 6
-609414.96049999    -1045194.222    -609420.4036   -1045157.2118
-609423.78489999   -1045137.4997    -609430.7512   -1045104.4406
    -609461.8814    -1045044.887    -609553.0165   -1044863.5194
#Sta/Elev= 30
       0  369.78   31.27  367.07   33.07  366.27   39.48   362.5   40.23  362.42
   44.13  359.81   44.54  359.04   44.59  357.75   45.31  355.55   47.35  355.37
   53.89  356.09   55.31  357.26   55.77  357.28   62.02  357.77   62.03  356.76
   63.43  356.55   64.18   358.1   81.51  358.03   98.41  358.41   193.3  358.25
   270.5   358.6  298.63  359.38  303.86  359.71  317.73  361.57  324.51  364.51
   326.8  364.77  328.62   365.8  346.91  368.43  356.85  371.77  361.37  369.68
#Mann= 3 ,-1 , 0
       0     .15       0   44.37     .05       0   55.44     .15       0
Levee=0,,,-1,61.97,357.76,,
#Block Obstruct= 1 ,-1
   153.9  155.72361.4517
Bank Sta=44.54,55.77
XS Rating Curve= 0 ,0
Exp/Cntr=0.3,0.1

Type RM Length L Ch R = 1 ,17782.89,62.55,62.87,61.97
XS GIS Cut Line= 4
    -609470.8038    -1045197.095-609477.57719999    -1045171.695
    -609480.4835   -1045126.6469    -609575.3674   -1044909.2278
#Sta/Elev= 30
       0  367.23   10.31  365.85   21.01  365.81   25.25  362.52   29.14  362.26
   33.12  356.58   46.79  356.14   48.18  354.63   53.26  354.63   54.36  355.91
   55.59  356.81   58.12   356.7   71.43  357.08   82.25  357.86   82.26  356.81
   86.78   356.7   87.64  357.27   88.13  357.77   93.12  357.71   95.37  357.51
  116.46  357.58  129.29  357.36  155.07  357.55  174.76  358.07  220.41  358.26
  236.89  358.58  283.05  360.03  297.17  360.74  301.47  360.81  308.65  361.26
#Mann= 3 , 0 , 0
       0     .15       0   46.79     .05       0   55.59     .15       0
#Block Obstruct= 2 ,-1
  123.33   138.2360.4653   60.62   69.08 359.908
Bank Sta=46.79,55.59
XS Rating Curve= 0 ,0
Exp/Cntr=0.3,0.1

Type RM Length L Ch R = 1 ,17720.02,5.95,5.94,5.93
XS GIS Cut Line= 6
-609530.90949999   -1045209.5616-609540.83509999   -1045177.0778
     -609541.896   -1045141.5778    -609542.1886   -1045093.1615
    -609613.9235   -1044959.6171    -609631.9701   -1044927.5846
#Sta/Elev= 30
       0  365.46   15.22  364.72   16.15  363.96   23.83  363.17   34.31  357.61
   41.52  357.02    49.5  357.51    52.4  358.81   52.43  356.79   52.61  355.32
   53.11  355.32   53.12  354.64   55.31  354.53   57.39  354.66   57.44  355.22
   57.94  355.34   60.19  354.69   64.31  354.67   64.44  355.31   64.91  355.32
   65.24  358.87    67.5  356.94  116.56  357.35  123.08  356.67  167.63  357.74
  242.81  357.93  254.77     360  278.34  373.07  292.67  373.29  306.28  370.34
#Mann= 3 ,-1 , 0
       0     .15       0    52.4     .04       0   65.24     .15       0
#Block Obstruct= 1 ,-1
  107.15  115.38360.2692
Bank Sta=52.4,65.24
XS Rating Curve= 0 ,0
Exp/Cntr=0.5,0.3

Type RM Length L Ch R = 1 ,17692.02,41.2,44.05,46.63
XS GIS Cut Line= 6
-609544.89559999   -1045215.8779-609568.07849999   -1045159.3655
-609569.86809999   -1045139.4457    -609584.1468   -1045094.0638
-609585.04899999   -1045083.2359-609645.95609999   -1044969.5427
#Sta/Elev= 30
       0  365.85    13.5   364.9   16.02  363.51   24.53  362.37   32.97  357.44
   43.75   356.7   51.15  356.45   51.73  355.95   52.11  356.46   54.11  356.24
   64.97  356.19   66.77  356.21   67.81  353.69   70.12  353.36   74.01  353.46
   75.45  353.71   77.54   356.2   112.1   356.1  127.58  356.28  133.49  356.79
  133.91  356.12   135.2  356.12  135.36  356.53   135.7     357  143.17  356.27
  152.93  356.95  211.03  356.88  228.34  357.09  241.83  357.04   268.5  371.35
#Mann= 3 ,-1 , 0
       0     .15       0   64.97    .045       0   77.71     .15       0
Bank Sta=66.77,77.54
XS Rating Curve= 0 ,0
Exp/Cntr=0.3,0.1

Type RM Length L Ch R = 1 ,17647.97,44.69,45.95,47.64
XS GIS Cut Line= 4
-609585.52739999   -1045225.4584-609605.14359999   -1045175.1529
-609621.57099999    -1045133.065    -609680.7776   -1044995.7996
#Sta/Elev= 30
       0  363.96    2.87  363.78    6.78   362.6    9.86  362.43   14.77  357.28
   43.32  355.93   59.51  354.85   70.15   355.4    70.4  352.86   77.31  352.98
   77.53  353.86    77.8  355.73   86.09  355.82   86.61  355.58   88.12  355.52
  120.47  356.19  140.44   356.2  147.34  356.31  148.56  356.72   157.2  356.33
  189.04  357.09  189.57  356.89  190.98  357.11   192.6  355.85  194.66  355.85
  195.62  356.72  225.89  356.55  237.22  357.06   240.2  357.46  248.66   362.3
#Mann= 3 , 0 , 0
       0     .15       0   70.15    .043       0    77.8     .15       0
#Block Obstruct= 2 ,-1
   32.55   43.62359.1464   53.99   67.02358.1605
Bank Sta=70.15,77.8
XS Rating Curve= 0 ,0
Exp/Cntr=0.3,0.1

Type RM Length L Ch R = 1 ,17556.69,44.71,42.68,40.34
XS GIS Cut Line= 2
    -609663.7304   -1045259.6598    -609765.9736   -1045040.7789
#Sta/Elev= 30
       0  362.56    3.89  362.45    17.2  360.62    28.1  359.88   29.15  358.88
    32.5  358.62   34.21  354.19    49.1  354.37   58.77  354.21   60.53  351.79
   66.87  352.11   70.34  354.93   82.63   354.9   83.15  354.41   83.69  354.83
   84.78   354.9   98.66  354.84  116.35   354.4  121.72  354.42  131.64   354.9
  134.28  355.49  153.96  355.67  177.53  355.21  214.78  355.38  224.11  355.63
  226.33  356.61   228.7  356.51  229.31  355.56     231  355.56  241.58  360.75
#Mann= 3 , 0 , 0
       0     .15       0   58.77     .04       0   70.34     .15       0
#Block Obstruct= 2 ,-1
   165.6  177.11358.3292       0   22.74 364.402
Bank Sta=58.77,70.34
XS Rating Curve= 0 ,0
Exp/Cntr=0.3,0.1

Type RM Length L Ch R = 1 ,17514.01,2.8,2.8,2.82
BEGIN DESCRIPTION:
17708  PF 227 ŽELEZNÝ MOSTEK V KVASINÁCH (F39)
END DESCRIPTION:
XS GIS Cut Line= 4
    -609698.4602   -1045261.8683     -609725.443   -1045231.8903
-609730.18059999   -1045212.4594-609799.52079999   -1045040.7983
#Sta/Elev= 30
       0  360.74   13.45  359.62   17.99  356.01   19.82  355.95   20.92  354.22
   42.05  354.32   45.47     355   47.45354.6392   47.81  352.09   48.83  351.72
   53.33  351.94   56.51  352.88   56.63  354.56   56.64   354.7   66.87  354.91
   74.05  354.08  108.73  354.29  128.22  355.11  154.53  354.58  168.29  355.23
  198.31  355.56  214.27  355.33  214.89  354.69  215.58  355.14  220.87  355.47
  223.59  356.93  226.48  356.46  227.14  355.57  228.65  355.57  245.47  364.99
#Mann= 3 ,-1 , 0
       0     .15       0   47.45     .04       0   56.63     .15       0
#Block Obstruct= 2 ,-1
   24.15   30.84357.4231   87.04   98.39357.2969
Bank Sta=47.45,56.64
XS Rating Curve= 0 ,0
Exp/Cntr=0.5,0.3

Type RM Length L Ch R = 1 ,17511.2 ,12.67,11.2,9.7
XS GIS Cut Line= 4
    -609701.1935   -1045262.4972-609728.17619999   -1045232.5193
-609732.91389999   -1045213.0884-609802.25409999   -1045041.4272
#Sta/Elev= 30
       0  360.67   11.61  359.75   17.21  355.79   18.74  355.74   19.88  354.22
   41.62  354.21   45.47     355   47.44  354.71   47.83  351.43   48.13  351.32
   53.04  351.69    56.5  352.85   56.64   354.7   61.45  354.49   66.63  354.89
   74.68  354.08  106.42  354.22  127.47  355.01  155.19  354.56  196.68  355.45
  212.48   355.3  212.49  354.98  213.78  354.89  215.01  355.32  220.24  355.33
  223.38  356.66  225.83  356.46   226.4  355.57  227.98  355.57  245.47  365.11
#Mann= 3 , 0 , 0
       0     .15       0   47.44     .04       0   56.64     .15       0
#Block Obstruct= 3 ,-1
   18.01   30.73358.0956   86.57   97.92357.2387  145.42  164.87357.8016
Bank Sta=47.44,56.64
XS Rating Curve= 0 ,0
Exp/Cntr=0.5,0.3

Type RM Length L Ch R = 1 ,17500.01,58,59.97,58.41
XS GIS Cut Line= 5
-609719.21379999    -1045277.659    -609734.1021   -1045261.8683
     -609740.789   -1045234.2777    -609742.4705   -1045214.3485
-609814.86039999   -1045044.8588
#Sta/Elev= 30
       0  361.64    7.38   361.6   20.08  354.36   38.77  353.85   57.64  353.87
   58.36  351.86   58.37  351.62   59.47   351.5   62.53  351.75   64.32  352.32
   67.25  354.44   67.66  354.52   74.65  354.81   80.73  354.56   85.77  354.08
   98.15  354.04  118.21  354.22   134.6  354.68  167.05   354.5  200.88  354.95
  220.42  354.81  220.99   354.5  221.74  354.99  226.68  355.39   229.5  356.42
  231.61  356.43  232.34  355.57  233.62  355.57  244.74  361.05  254.39  366.16
#Mann= 3 , 0 , 0
       0     .15       0   57.64     .04       0   67.66     .15       0
#Block Obstruct= 3 ,-1
   49.69   56.55356.8469   93.82  105.17357.1008  152.62  172.07357.6448
Bank Sta=57.64,67.66
XS Rating Curve= 0 ,0
Exp/Cntr=0.3,0.1

Type RM Length L Ch R = 1 ,17440.04,41.3,46.93,51.33
XS GIS Cut Line= 4
-609760.83949999    -1045326.651-609797.06219999   -1045248.2126
    -609803.9891   -1045215.1089    -609864.0548   -1045079.3023
#Sta/Elev= 29
       0  357.96   25.55   358.3   31.64  355.71   35.65  353.91   45.53  353.87
   57.03  353.52   66.93  353.77   89.06  353.62  103.17  353.11   103.2  352.94
  104.02  350.75  110.53  350.85  112.14  353.96  120.22   353.9  121.54  353.76
  147.61  353.53  159.11  353.67     172  354.09  184.58   354.4  239.73  354.43
  240.01  354.29  245.36  353.92  251.56  354.58  254.38  356.22  257.06  356.15
  257.65  355.59   259.2  355.59  261.12   356.6  268.72  361.06
#Mann= 3 , 0 , 0
       0     .15       0  103.17     .04       0  112.14     .15       0
Levee=-1,76.04,353.71,-1,114.49,353.85,,
#Block Obstruct= 4 ,-1
       0   17.78361.0793  182.05  227.99357.3547  138.13  160.15356.6496
   91.36  102.14356.3394
Bank Sta=103.17,112.14
XS Rating Curve= 0 ,0
Exp/Cntr=0.3,0.1

Type RM Length L Ch R = 1 ,17393.11,13.26,15.1,14.97
XS GIS Cut Line= 5
    -609773.9127   -1045343.0054    -609816.9842   -1045291.5139
-609843.09259999   -1045243.5518-609853.51619999   -1045227.0443
    -609891.0705   -1045107.7374
#Sta/Elev= 30
       0   357.3    4.31  355.16   28.77  355.07   35.81  355.35   38.43  354.22
   52.76  353.59   67.02  353.62   83.96   353.1   99.99  353.33  120.87  353.04
  123.95   352.8   126.5  350.88  132.18  350.89  132.74  352.01  132.96  353.19
  160.85  353.79  180.88  353.98  182.01  353.81  183.61  354.08  226.35  354.59
  242.41  354.53  248.19  354.04   251.2   354.3  256.76   354.1  257.29  353.76
   259.3  354.27  261.37  354.34  263.58  356.12  264.05  355.92  266.34     356
#Mann= 3 , 0 , 0
       0     .15       0  120.87     .04       0  132.96     .15       0
Levee=-1,117.96,353.22,0,,,,
#Block Obstruct= 2 ,-1
   52.09    52.9356.6096   67.13    78.1356.4224
Bank Sta=120.87,132.96
XS Rating Curve= 0 ,0
Exp/Cntr=0.3,0.1

Type RM Length L Ch R = 1 ,17378   ,2.96,2.99,2.78
XS GIS Cut Line= 6
     -609777.842   -1045343.8274-609812.85159999     -1045322.95
    -609833.5683   -1045281.9181    -609866.1356    -1045237.247
    -609898.0165   -1045115.3894    -609907.0396   -1045097.3429
#Sta/Elev= 30
       0  356.33    4.12  355.13   40.29   354.5   59.87  353.74   93.02  353.51
   96.51  353.21  118.31  353.47  127.69  353.97  128.16  353.84  128.17  353.23
  128.18  351.66  132.69  350.83  135.79  351.67  135.87  353.64   135.9  353.74
  136.49  353.96   151.3  353.38  175.95  353.43  192.67  353.57  193.59  353.99
  195.42  354.03  247.07  354.26  263.29  353.47  267.08  354.21  269.69  355.94
  271.77  356.02  272.35  355.51  273.92  355.51  280.14  359.06  288.57  364.44
#Mann= 3 ,-1 , 0
       0     .15       0  128.43     .04       0  136.02     .15       0
Levee=-1,127,353.97,-1,136.06,353.99,,
#Block Obstruct= 4 ,-1
   164.3  174.89356.4578  180.57  187.88356.5107   217.5   225.9357.2125
  236.65  247.52 357.206
Bank Sta=127.69,135.9
XS Rating Curve= 0 ,0
Exp/Cntr=0.5,0.3

Type RM Length L Ch R = 1 ,17375.01,8.74,9.01,9.67
XS GIS Cut Line= 6
    -609780.0582   -1045345.8438    -609815.0678   -1045324.9665
-609835.78449999   -1045283.9345-609868.35179999   -1045239.2635
    -609900.2327   -1045117.4058     -609909.256   -1045099.3593
#Sta/Elev= 30
       0  356.66    1.51  356.22     3.8  353.94   13.71  354.17   20.31   353.8
   42.47  353.75   45.33  354.19   54.28  353.43   87.05  353.15   94.83  352.77
   101.2  353.43  113.33  353.34  128.45  353.89  128.49  352.43   128.5  351.65
  133.03  350.82  136.13  351.64   136.2  353.67  136.26  353.93  152.01  353.35
  194.94  353.56  195.97  354.01  248.13  354.18  263.75  353.46  267.91  354.19
  270.65  355.98  272.83  356.06  273.43  355.51  275.01  355.51  288.57  363.86
#Mann= 3 , 0 , 0
       0      .1       0  128.45     .04       0  136.26      .1       0
Levee=-1,126.27,353.8,0,,,,
#Block Obstruct= 3 ,-1
  165.99  176.58 356.446  182.19   189.5356.5049  218.36  248.38357.1706
Bank Sta=128.45,136.26
XS Rating Curve= 0 ,0
Exp/Cntr=0.5,0.3

Type RM Length L Ch R = 1 ,17366   ,28.61,25.35,19.86
XS GIS Cut Line= 5
    -609829.4397   -1045357.2129    -609861.4726   -1045259.9622
    -609876.1358   -1045246.3611    -609880.4211   -1045229.0826
    -609907.8099   -1045124.7443
#Sta/Elev= 30
       0  365.52   12.38  355.09   21.35  353.94   23.66  353.65    37.8  353.23
    61.6   352.8    72.7  352.91   79.98  353.14   80.52  353.26   80.93  352.56
   82.58   352.5    82.9  353.53    83.5   353.6   89.54  353.39   101.6  352.66
  106.24  352.26  108.13  351.52  111.97  350.79  116.19  351.52  116.56  353.71
   122.6  353.39  139.25   353.2  154.31   353.4  182.83  353.52  184.41  354.03
  217.23  354.12  232.88  354.01  244.41  353.58   245.3  353.44  248.07  353.81
#Mann= 3 , 0 , 0
       0      .1       0   101.6    .035       0  116.56      .1       0
Levee=-1,84.01,353.38,0,,,,
#Block Obstruct= 3 ,-1
   65.59   77.29355.9429  121.07  132.79 356.422  224.73  231.42357.0443
Bank Sta=101.6,116.56
XS Rating Curve= 0 ,0
Exp/Cntr=0.3,0.1
