HEC-RAS study PPO_Kvasiny_efektiv.prj: PPO_Kvasiny_efektivita

--- PPO_Kvasiny_efektiv.g08 (geometry) --- (continued)

Type RM Length L Ch R = 1 ,18658.06,22,33.51,26.87
XS GIS Cut Line= 6
-608811.08549999    -1044755.116     -608825.589   -1044701.0257
    -608807.8792   -1044691.7325-608803.30299999   -1044664.7705
    -608806.6867   -1044622.1356-608834.09479999   -1044582.8844
#Sta/Elev= 30
       0  378.22   12.72  374.61   27.41  371.22   36.15  368.78    43.1  367.32
    46.5  365.69   53.84  365.69   56.09  365.96   61.11  366.23   62.71   366.9
   62.73  364.21   69.51  364.09   70.75  365.09   74.46366.5206   77.86  366.86
   92.64  366.97   96.45  367.35  103.66  367.39  122.92   366.9  134.34  367.11
  137.58  367.24   142.8367.2064  146.19  367.18  147.55  366.45  148.03  366.83
  150.17  367.09  151.31  366.42  171.67  379.13  183.96  386.99  194.08  389.02
#Mann= 5 ,-1 , 0
       0      .2       0   62.71    .045       0   74.46     .12       0
  134.34     .05       0   142.8     .12       0
Levee=-1,62.62,366.83,-1,137.53,367.18,,
#Block Obstruct= 1 ,-1
  104.88  123.34370.1295
Bank Sta=62.71,74.46
XS Rating Curve= 0 ,0
Exp/Cntr=0.3,0.1

Type RM Length L Ch R = 1 ,18624.55,27.54,38.49,47.2
XS GIS Cut Line= 6
    -608813.3292   -1044757.0751-608830.65819999   -1044713.3605
     -608838.708   -1044671.6675    -608829.9133   -1044663.7088
    -608830.5483   -1044653.6758    -608851.3869   -1044598.6741
#Sta/Elev= 30
       0  378.92   15.14  374.94   22.67  373.16    30.2  371.61   40.84  368.61
   44.87  368.72   44.88  367.19   46.46  365.77   56.35  365.59   58.15  365.81
   71.85  365.45   85.93  366.54   89.66  367.02   89.67  364.06   98.15  364.03
   101.2  367.01  101.96   366.9  120.26  367.04  122.19  365.97  123.18  366.43
  124.31  367.04  129.18  367.16  132.12  367.14  133.58  366.63  136.31  368.67
  144.85  374.62  152.76  379.57  161.81  385.47  167.38  386.49  170.22  387.15
#Mann= 5 ,-1 , 0
       0      .2       0   89.66     .05       0   101.2     .12       0
  123.18     .05       0  133.58     .15       0
Levee=-1,88.75,366.79,-1,105.8,366.93,,
#Block Obstruct= 2 ,-1
   43.76   47.02 370.226   55.44   78.67 370.226
Bank Sta=89.66,101.2
XS Rating Curve= 0 ,0
Exp/Cntr=0.3,0.1

Type RM Length L Ch R = 1 ,18495.51,25.6,24.88,23.57
XS GIS Cut Line= 4
    -608887.9529   -1044774.1613    -608917.6792   -1044750.0879
    -608934.0835    -1044737.917    -608970.0669   -1044707.7544
#Sta/Elev= 27
       0  370.29    6.96  368.39   10.03  368.32   13.09  368.15   15.21  365.51
   21.57  365.46   28.43  365.09   37.14  365.48   42.19  365.61   44.14   362.6
   47.66  362.74   49.82   364.1   51.54  364.96   53.01  365.07   58.45     365
   67.51  370.43    69.1  370.93    70.8  371.82   71.62   371.9   74.81   373.6
    79.7  375.88   86.45  376.34   91.06   376.8  100.25  377.07  101.89  377.02
  102.68  377.63  105.63  377.96
#Mann= 4 ,-1 , 0
       0      .2       0   42.19    .045       0   51.54     .05       0
   58.45      .2       0
#Block Obstruct= 1 ,-1
   16.66   42.27367.0693
Bank Sta=42.19,51.54
XS Rating Curve= 0 ,0
Exp/Cntr=0.3,0.1

Type RM Length L Ch R = 1 ,18350.04,2,2,2.21
XS GIS Cut Line= 4
    -608978.2241   -1044895.2065    -609008.2817   -1044865.0536
-609022.72899999   -1044851.2234-609048.56549999   -1044818.2857
#Sta/Elev= 22
       0  373.57     9.6  371.52   13.82  370.74   28.98  366.75   29.65  366.55
    33.8  363.79   35.16  363.25   36.75   362.9   47.26  363.08    47.8  362.16
   49.92  361.34   52.39  361.21   55.13  361.42    56.2  361.99   57.62  363.12
   57.71  363.12   59.38  363.15    65.2     363    67.3  363.14   75.51  363.06
   96.41  364.13  104.44  364.33
#Mann= 4 ,-1 , 0
       0      .1       0   47.26     .05       0   57.71     .06       0
    67.3     .15       0
Bank Sta=47.26,57.71
XS Rating Curve= 0 ,0
Exp/Cntr=0.5,0.3

Type RM Length L Ch R = 3 ,18348.94,,,
BEGIN DESCRIPTION:
NOVE NAVRHOVANA LAVKA
END DESCRIPTION:
Bridge Culvert--1,0,-1,-1, 0
Deck Dist Width WeirC Skew NumUp NumDn MinLoCord MaxHiCord MaxSubmerge Is_Ogee
0.2,1.5,1.4,0, 7, 7, , , 0.98, 0, 0,0,,
   46.75   47.56   50.02   52.47   54.93   57.38   58.19
  363.62   363.9  364.32  364.47  364.32   363.9  363.62
       0  363.22  364.01  364.15  364.01  363.22       0
    46.3   47.11   49.57   52.02   54.48   56.93   57.74
  363.62   363.9  364.32  364.47  364.32   363.9  363.62
       0  363.22  364.01  364.15  364.01  363.22       0
BR Coef=-1 , 0 , 0 ,, 0 ,,,0.8,-1,,0,
WSPro=,,,, 1 ,,,, 0 ,,,, 0 ,,,,-1 ,-1 ,-1 , 0 , 0 , 0 , 0 , 0
BC Design=,, 0 ,, 0 ,,,,,,
BC Use User HTab Curves=0
BC User HTab FreeFlow(D)= 0

Type RM Length L Ch R = 1 ,18348.04,7.11,6.87,7.11
XS GIS Cut Line= 4
    -608980.1664   -1044896.0904     -609009.671   -1044866.4922
-609024.11829999    -1044852.662-609051.48649999   -1044819.8097
#Sta/Elev= 22
       0   373.3    6.85  371.83   14.58  370.39   27.13  367.13   31.91  364.08
   32.82  363.72   33.93  363.69   37.54  362.88   47.11  363.08   47.12  362.22
    47.3  362.08   49.13  361.33   51.22  361.18   54.38  361.41   56.87   362.8
   58.56  363.11   64.54  362.98   66.68  363.12   71.95  363.09   74.49  362.95
   94.77  364.01  104.55  364.23
#Mann= 4 ,-1 , 0
       0      .1       0   47.11     .05       0   58.56     .07       0
   71.95     .15       0
Bank Sta=47.11,58.56
XS Rating Curve= 0 ,0
Exp/Cntr=0.5,0.3

Type RM Length L Ch R = 1 ,18341.17,3.64,3.82,3.48
XS GIS Cut Line= 3
    -608984.7855   -1044901.5539    -609031.6963   -1044854.4518
    -609056.4353   -1044826.8159
#Sta/Elev= 22
       0  372.94    2.13  372.61   20.54  369.17   21.45  368.93   21.89  368.65
   33.77  363.06   39.86  362.88   43.25  362.84   46.71  362.94   47.49  362.85
   49.56  361.32   51.05  361.09   54.92  361.34    57.3  362.81   59.63  363.03
   65.57  362.92   66.48  362.98   67.49  363.04   74.34  362.62   81.72  362.96
   86.35  363.35  103.57  363.97
#Mann= 4 ,-1 , 0
       0      .1       0   47.49     .05       0    57.3     .07       0
   66.48     .15       0
Bank Sta=47.49,57.3
XS Rating Curve= 0 ,0
Exp/Cntr=0.3,0.1

Type RM Length L Ch R = 1 ,18337.36,14.84,14.42,14.55
XS GIS Cut Line= 4
     -608988.397   -1044905.6744    -609016.6957   -1044874.6581
-609031.05539999   -1044860.7368-609065.50409999   -1044820.1635
#Sta/Elev= 23
       0  372.66    7.27  371.71   18.26  369.64   22.38  369.43   23.75  366.65
   32.89  362.99   44.01  362.82   47.08  362.88   47.98  362.78   49.83  361.33
   51.34  361.04   55.16  361.22   56.57  362.09   57.45  362.74   60.24  362.98
   66.23  362.88   67.23  362.95   74.45  362.47   84.01  362.91   87.64  363.22
  100.82  363.72  111.88  364.06  115.21  364.08
#Mann= 4 ,-1 , 0
       0      .1       0   47.98     .05       0   57.45     .07       0
   67.23     .15       0
#Block Obstruct= 1 ,-1
   28.28   43.46366.8377
Bank Sta=47.98,57.45
XS Rating Curve= 0 ,0
Exp/Cntr=0.3,0.1

Type RM Length L Ch R = 1 ,18322.93,16.56,16.4,16.08
XS GIS Cut Line= 2
    -608999.2052   -1044914.5843-609092.44469999   -1044816.5633
#Sta/Elev= 30
       0   371.6    1.44  371.41   11.32  370.72   17.22  369.69      22  369.71
   22.18  369.37   26.56  363.14   26.79  363.06   32.25  362.96   36.52  363.02
   46.17  362.61   46.51  362.42    46.8  362.39   48.27   361.2   49.96  360.97
   52.55  361.04   54.13  361.21   56.24  362.84   58.62  362.74   59.86  362.85
   65.92  362.78   67.09  362.35   68.75  362.34    85.2  362.75  103.25  363.53
   109.5  363.69  124.02  363.67  125.26  364.47   130.6   365.3  135.28  366.61
#Mann= 4 ,-1 , 0
       0      .1       0   46.17     .05       0   56.24     .07       0
   65.92     .15       0
#Block Obstruct= 1 ,-1
   26.73   35.54366.0181
Bank Sta=46.17,56.24
XS Rating Curve= 0 ,0
Exp/Cntr=0.3,0.1

Type RM Length L Ch R = 1 ,18306.53,11.47,11.55,11.69
XS GIS Cut Line= 3
-609011.42359999   -1044926.7722     -609089.892   -1044841.4859
-609102.89469999   -1044819.0525
#Sta/Elev= 28
       0  371.18    6.19  370.79   12.56  370.67   15.64  369.97   21.26   369.1
   27.95  363.31   28.33  363.04    42.1  362.52   42.75  362.52   42.97  362.64
   43.45  362.63   46.81  362.42   47.74  361.76   48.31  361.11   49.74  361.06
   55.15  361.16   56.14  361.95   56.76  362.86   61.31   362.7   67.32  362.66
   68.74  361.99   85.01  362.37   97.26  363.06  115.89  363.41  131.24  363.56
  131.94  364.19  136.75  364.86  141.82  366.12
#Mann= 4 ,-1 , 0
       0      .1       0   46.81     .05       0   56.76     .07       0
   67.32     .15       0
#Block Obstruct= 2 ,-1
   39.21   42.75365.5524   76.18   94.88 365.575
Bank Sta=46.81,56.76
XS Rating Curve= 0 ,0
Exp/Cntr=0.3,0.1

Type RM Length L Ch R = 1 ,18294.98,16.32,15.92,15.19
XS GIS Cut Line= 4
    -609019.4125   -1044934.5905    -609077.4164   -1044872.4435
    -609103.2397   -1044839.8467    -609108.1081   -1044820.1617
#Sta/Elev= 29
       0  370.98    4.19  370.91   17.42  370.05   20.37  369.57   23.32  368.91
   26.83  366.55   34.78   362.5    43.3  362.56   47.13  362.35   48.05  361.28
    48.1  361.13   51.66  361.15   55.02  361.06   55.67  361.07   55.85  361.23
   56.87  362.72   61.37  362.59   68.21  362.57   69.87  361.74   76.63   361.9
   81.35  362.14   84.78  362.13   90.37  362.32  106.65  363.15  129.28  363.42
  136.27  363.36  136.81  363.82  142.18  364.59  146.87  365.89
#Mann= 4 ,-1 , 0
       0      .1       0   47.13     .05       0   56.87     .07       0
   68.21     .15       0
Bank Sta=47.13,56.87
XS Rating Curve= 0 ,0
Exp/Cntr=0.3,0.1

Type RM Length L Ch R = 1 ,18279.06,5.31,5.32,5.33
BEGIN DESCRIPTION:
PETRUV JEZ (NADJEZI)
END DESCRIPTION:
XS GIS Cut Line= 5
-609032.27279999   -1044946.5812    -609059.4153   -1044915.6818
     -609083.818   -1044887.4375-609116.26419999   -1044848.5425
-609124.47399999   -1044813.5362
#Sta/Elev= 30
       0  372.24     1.5  372.25   15.72  369.87   19.55  369.35   23.91  369.19
   26.11  368.71   29.13  368.34   32.56  365.49   35.93  362.09   43.99  362.42
   46.63  362.26   46.82   362.2   46.87  361.22   54.47  361.12   56.67  361.33
   56.72  361.94   56.73  362.29   62.98  362.49   69.03  362.46   70.79   361.7
   84.14  361.98   95.28  362.05  101.69  362.42  106.65  362.88  137.65  363.14
  143.62  362.91     144  363.26  151.97   364.2  157.22  365.52  165.06  367.28
#Mann= 4 ,-1 , 0
       0      .1       0   46.63     .05       0   56.73     .07       0
   69.03     .15       0
#Block Obstruct= 1 ,-1
    85.1  103.82365.3277
Bank Sta=46.63,56.73
XS Rating Curve= 0 ,0
Exp/Cntr=0.3,0.1

Type RM Length L Ch R = 1 ,18273.75,10.28,9.7,8.84
XS GIS Cut Line= 5
    -609036.4443   -1044949.8598-609064.65399999   -1044917.7456
-609089.05669999   -1044889.5013-609120.98169999   -1044852.9628
    -609132.1506   -1044815.9045
#Sta/Elev= 30
       0  371.64     5.2  371.19   16.67   369.3   21.28  367.85      29  367.62
   33.77  364.43   35.92  362.28   38.55  362.42   46.23  362.26   46.25  361.49
   46.94   361.5   47.36  360.55   47.57   360.6   47.98  359.05   48.96  359.47
   52.34  359.56    57.2  360.29   57.82  362.19   62.85  362.44    68.5  362.42
   68.85  362.41   70.63  361.65   94.71   362.2  104.69  362.78  125.75   363.1
  141.77  363.11  145.94  362.92  146.35  363.21  157.05   364.3   167.3  366.38
#Mann= 4 ,-1 , 0
       0      .1       0   46.23     .04       0   57.82     .07       0
    68.5     .15       0
#Block Obstruct= 1 ,-1
   86.04  104.85365.4245
Bank Sta=46.23,57.82
XS Rating Curve= 0 ,0
Exp/Cntr=0.3,0.1

Type RM Length L Ch R = 1 ,18264.04,12.48,12.71,12.7
XS GIS Cut Line= 5
    -609043.6799   -1044956.0504    -609072.4114   -1044924.5346
-609084.51969999   -1044908.6165    -609125.8273   -1044857.4816
-609142.94559999   -1044817.4285
#Sta/Elev= 30
       0  370.31   12.28  369.16   15.21  368.69   17.39   367.5   25.74  366.82
    37.8  361.96   41.05  362.18   45.27  362.15   46.56  361.95   47.29  361.26
   47.47   360.3   49.85  360.35   53.13   360.2   57.68  360.44   58.07  361.27
   59.09   362.2   63.06  362.35   68.94  362.33   70.89  361.61    72.5  361.89
   88.18  361.87   88.96  362.28   90.18  362.38  112.24  362.77  146.92  363.09
  148.75  362.97  149.04  363.13  153.37  363.53  164.13  364.28  171.94  365.37
#Mann= 4 ,-1 , 0
       0      .1       0   45.27     .05       0   59.09     .07       0
   68.94     .15       0
Bank Sta=45.27,59.09
XS Rating Curve= 0 ,0
Exp/Cntr=0.3,0.1

Type RM Length L Ch R = 1 ,18224.5 ,18.07,18.46,18.77
XS GIS Cut Line= 3
    -609075.6612   -1044979.0075    -609117.0775    -1044932.579
-609210.79199999   -1044805.8233
#Sta/Elev= 28
       0  365.11   10.49  364.17   13.68  363.68   26.24  362.67   41.24  362.03
   43.28     362   43.96  361.76   46.43  360.03   48.49  359.94    55.2  360.03
   57.34  361.78   66.26  361.87   67.31  360.99   68.09  361.51   70.76  361.49
   84.16  361.75   86.64  361.61    87.3  361.49      90  361.78   102.4  362.52
  108.88  362.59  158.83  362.54  177.06  362.44  196.05  362.67  204.95  363.03
  214.11  363.16  215.94  363.32  219.85  363.87
#Mann= 4 ,-1 , 0
       0      .1       0   43.28     .05       0   57.34     .07       0
   66.26      .2       0
#Block Obstruct= 1 ,-1
   17.57   28.26365.9847
Bank Sta=43.28,57.34
XS Rating Curve= 0 ,0
Exp/Cntr=0.3,0.1

Type RM Length L Ch R = 1 ,18206.04,5.09,4.98,4.99
XS GIS Cut Line= 4
     -609080.951    -1044998.105    -609116.2027    -1044960.872
    -609129.9171   -1044946.3148-609272.49179999   -1044770.8857
#Sta/Elev= 30
       0  367.22    4.83  366.36    6.94  366.52    8.97  365.99   12.57   364.3
   14.78  363.49   28.27  362.63   55.41   362.2   55.65  361.65      56  359.96
    58.7  359.69   63.69  359.58   65.74  359.86   65.96  360.26   66.01  361.53
   66.11  361.55   66.12   361.7   68.84  361.82   77.27  361.64    78.3  360.92
   79.13  361.48   90.93  361.17  129.25   362.2  170.35  361.86     247  362.15
  252.55  362.43  264.74  363.43  279.08  365.99   280.2  366.37  297.33  368.69
#Mann= 4 ,-1 , 0
       0      .1       0   55.41     .05       0   66.12     .07       0
   77.27      .2       0
Bank Sta=55.41,66.12
XS Rating Curve= 0 ,0
Exp/Cntr=0.5,0.3

Type RM Length L Ch R = 1 ,18201.06,23.86,23.02,22.09
XS GIS Cut Line= 4
     -609081.967   -1045006.5717-609120.09479999    -1044964.001
    -609133.8092   -1044949.4436    -609276.3839   -1044774.0146
#Sta/Elev= 30
       0  370.45     4.8  370.18    9.09  368.12   16.22  367.74   26.16  363.16
    34.1  362.62   38.88  362.59   49.59  362.04   61.21  362.12   61.43  361.72
   62.15  359.61   63.21   359.5   70.02  359.52   70.68  359.73   71.92  361.91
   83.07  361.59   84.04  360.91   84.84  361.47   94.82  361.15  102.39  361.66
  115.93  361.61  134.35  362.12  200.36  361.64   211.5   361.1  215.58  361.35
  219.39     362  259.37  362.04  269.05  363.42  272.69  363.62  303.21  368.19
#Mann= 4 ,-1 , 0
       0     .15       0   61.21     .05       0   71.92     .07       0
   83.07      .2       0
Levee=0,,,-1,133.77,362.12,,
#Block Obstruct= 1 ,-1
    3.93   17.13371.7588
Bank Sta=61.21,71.92
XS Rating Curve= 0 ,0
Exp/Cntr=0.5,0.3

Type RM Length L Ch R = 1 ,18178.04,32.9,33.23,33.2
XS GIS Cut Line= 4
    -609103.6508   -1045021.0811-609138.55079999   -1044978.8772
    -609151.1605   -1044963.3531    -609291.7859   -1044770.6855
#Sta/Elev= 30
       0  370.22    4.28  368.69   21.67  367.17   22.82  366.86   27.24  364.45
   32.28  364.28    34.4  363.32   47.53  361.85   54.36  361.67   56.22360.7247
   59.04  359.39   62.85  359.24   66.74  359.62   67.19  359.89   73.29 361.474
   73.82  361.58   80.03  361.53   80.86  360.85   81.81  361.33  116.27  361.85
  148.98  361.84   172.7  361.43   230.3  361.73  231.77  361.18  233.41  361.85
   264.6  361.63  270.94  361.97  275.13  361.92  301.82  367.24  313.29   368.9
#Mann= 3 ,-1 , 0
       0     .15       0   56.22     .05       0   73.29     .15       0
Levee=0,,,-1,115.79,361.81,,
#Block Obstruct= 1 ,-1
  115.17  115.55 364.834
Bank Sta=54.36,73.82
XS Rating Curve= 0 ,0
Exp/Cntr=0.3,0.1

Type RM Length L Ch R = 1 ,18070.04,26.03,25.34,24.56
XS GIS Cut Line= 4
    -609188.4695   -1045088.7556-609221.08839999   -1045048.4074
    -609233.1209    -1045032.432    -609365.3255   -1044814.4483
#Sta/Elev= 30
       0     370   10.54  368.86   20.03  368.66   33.14  367.11   37.84  365.32
   47.64  364.27    53.9360.3909   56.53  358.81   58.19  358.78    58.7  358.34
   59.86  358.27   62.11  358.56   65.23  358.46   66.45  358.77   66.61  360.22
   77.76  360.33   80.25   360.6   86.85  360.61   96.19  360.93  140.38  360.59
  183.97  360.75  216.94  360.42  239.52  360.42  240.85  359.79  242.33  360.48
  260.41  360.53  271.53  360.28  299.39  361.45  320.98  363.85  326.83  364.34
#Mann= 3 ,-1 , 0
       0     .15       0    53.9     .05       0   66.61     .15       0
Levee=0,,,-1,96.59,360.86,,
#Block Obstruct= 1 ,-1
   94.75  105.86363.8593
Bank Sta=53.9,66.61
XS Rating Curve= 0 ,0
Exp/Cntr=0.3,0.1

Type RM Length L Ch R = 1 ,18044.69,39.68,37.85,34.98
XS GIS Cut Line= 4
    -609211.3246   -1045101.1375    -609241.9703   -1045063.7315
    -609258.5068   -1045037.9345    -609384.8456   -1044831.5591
#Sta/Elev= 30
       0  369.31    2.39  369.32   19.27  368.35   22.94  368.32   23.29  367.96
   25.53  366.85   30.81  366.28   34.45  366.19   44.62  364.96   48.36  361.71
   52.05  358.11   60.57  358.01   60.99  358.01      61  360.18   63.04  359.73
   89.32  360.45  107.65  360.45   114.4  360.28  170.26  360.44  187.43  360.13
  198.58  360.24  215.58  360.05  239.86  360.35  241.36  359.56  242.68  360.34
  258.25  360.37  270.11  359.83  275.91   360.3  293.32  360.54  320.97  362.15
#Mann= 3 , 0 , 0
       0     .15       0   48.36     .05       0      61     .15       0
Levee=0,,,-1,107.71,360.41,,
#Block Obstruct= 4 ,-1
   69.09   78.84363.0494   36.85   45.32 368.134  320.66  320.97365.1357
  299.39  309.67364.1195
Bank Sta=48.36,61
XS Rating Curve= 0 ,0
Exp/Cntr=0.3,0.1

Type RM Length L Ch R = 1 ,17958.03,4.98,4.96,5.01
XS GIS Cut Line= 5
-609289.07889999   -1045149.6626    -609326.2672   -1045090.5068
    -609331.3531   -1045071.1643-609362.16739999   -1045001.6811
     -609463.228   -1044828.8855
#Sta/Elev= 30
       0  369.29   10.49  367.12   14.99  366.62   22.52  362.14   25.14  361.66
   48.53   359.5   60.23  359.41   60.84  358.54   61.76  359.58   70.13  359.78
   75.55 359.302    75.8   359.3   75.82  357.91   79.63  357.53    84.3  357.64
   84.42  358.13   85.85  358.13   85.91  359.33   86.02359.3391   88.33  359.73
  100.05  359.74  101.16  359.17  113.29  359.09  128.04  359.49  246.69  359.43
  300.86  359.83  339.45  361.39  344.75  362.14  352.79  362.59  366.06  364.66
#Mann= 3 ,-1 , 0
       0     .15       0   75.55     .04       0   86.02     .15       0
Levee=-1,70.67,359.7,-1,88.68,359.7,,
#Block Obstruct= 1 ,-1
   137.4   140.4362.4691
Bank Sta=75.55,86.02
XS Rating Curve= 0 ,0
Exp/Cntr=0.5,0.3

Type RM Length L Ch R = 1 ,17953.06,18.09,19.04,21.99
XS GIS Cut Line= 5
    -609293.7773   -1045151.3166    -609330.9657   -1045092.1607
    -609336.0515   -1045072.8183    -609366.8658   -1045003.3351
-609467.92639999   -1044830.5395
#Sta/Elev= 30
       0  369.07    11.2  366.99   16.25  366.54   23.81  361.64   31.67  361.21
   34.54  359.98   49.71  359.02   55.47  359.16   56.39  358.03   57.93  359.51
   75.67   359.3   75.68  357.75   75.77  357.73   83.46  357.58   84.45  357.61
   84.51  358.04   86.02  357.94   86.03  358.73   86.12  358.74   86.13  359.33
   88.09  359.64  117.88  359.15     130   359.5  300.62  359.77  332.39     361
  334.26  362.21  336.13  362.19  336.58  361.57  354.75  362.83  366.06  365.13
#Mann= 3 , 0 , 0
       0     .15       0   75.67     .04       0   86.13     .15       0
Levee=-1,66.05,359.48,-1,89.61,359.48,,
Bank Sta=75.67,86.13
XS Rating Curve= 0 ,0
Exp/Cntr=0.5,0.3

Type RM Length L Ch R = 1 ,17934.03,65.98,74.44,72.11
XS GIS Cut Line= 5
    -609319.7439   -1045164.6074-609346.21489999    -1045097.348
    -609356.5102   -1045080.2014-609385.44929999   -1045009.9555
    -609484.1037    -1044838.313
#Sta/Elev= 30
       0  369.98    4.24  370.22     6.8  369.31   10.23  368.96   10.42  368.14
    18.3  367.33   23.78   362.9   27.99   362.3   36.51  359.32   52.99   358.4
   54.67  357.65   57.58  359.02   76.56   358.8   78.51  357.62   84.98  357.26
   85.93  357.35    88.7358.8978   94.07  359.24  120.45  358.94  180.97   359.7
   185.5  359.25  295.12  359.45   312.5  360.15  328.34  360.25  331.09  361.19
  343.38  361.45  347.01  361.72  352.88  362.67   359.2  364.58  366.23  367.65
#Mann= 3 ,-1 , 0
       0     .15       0   76.56     .04       0    88.7     .15       0
Levee=0,,,-1,94.23,359.25,,
#XS Ineff= 2 , 0
           66.97  361.58
Permanent Ineff=
       F       F
Bank Sta=76.56,88.7
XS Rating Curve= 0 ,0
Exp/Cntr=0.3,0.1

Type RM Length L Ch R = 1 ,17840.02,57.92,57.13,54.77
XS GIS Cut Line= 6
-609414.96049999    -1045194.222    -609420.4036   -1045157.2118
-609423.78489999   -1045137.4997    -609430.7512   -1045104.4406
    -609461.8814    -1045044.887    -609553.0165   -1044863.5194
#Sta/Elev= 30
       0  369.78   31.27  367.07   33.07  366.27   39.48   362.5   40.23  362.42
   44.37  359.45   44.54  359.04   44.59  357.75   45.31  355.55   47.35  355.37
   53.89  356.09   55.44357.2657   62.02  357.77   62.03  356.76   63.43  356.55
   63.75  357.01   64.18   358.1   81.51  358.03   98.41  358.41   193.3  358.25
   270.5   358.6  298.63  359.38  303.86  359.71  317.73  361.57  324.51  364.51
   326.8  364.77  328.62   365.8  346.91  368.43  356.85  371.77  361.37  369.68
#Mann= 3 ,-1 , 0
       0     .15       0   44.37     .05       0   55.44     .15       0
Levee=0,,,-1,66.05,357.88,,
#Block Obstruct= 1 ,-1
   153.9  155.72361.4517
Bank Sta=44.54,55.44
XS Rating Curve= 0 ,0
Exp/Cntr=0.3,0.1

Type RM Length L Ch R = 1 ,17720.02,5.95,5.94,5.93
XS GIS Cut Line= 6
-609530.90949999   -1045209.5616-609540.83509999   -1045177.0778
     -609541.896   -1045141.5778    -609542.1886   -1045093.1615
    -609613.9235   -1044959.6171    -609631.9701   -1044927.5846
#Sta/Elev= 30
       0  365.46   15.22  364.72   16.15  363.96   23.83  363.17   34.31  357.61
   41.52  357.02    49.5  357.51    52.4  358.81   52.43  356.79   52.61  355.32
   53.11  355.32   53.12  354.64   55.31  354.53   57.39  354.66   57.44  355.22
   57.94  355.34   60.19  354.69   64.31  354.67   64.44  355.31   64.91  355.32
   65.24  358.87    67.5  356.94  116.56  357.35  123.08  356.67  167.63  357.74
  242.81  357.93  254.77     360  278.34  373.07  292.67  373.29  306.28  370.34
#Mann= 3 ,-1 , 0
       0     .15       0    52.4     .04       0   65.24     .15       0
#Block Obstruct= 1 ,-1
  107.15  115.38360.2692
Bank Sta=52.4,65.24
XS Rating Curve= 0 ,0
Exp/Cntr=0.5,0.3

Type RM Length L Ch R = 1 ,17692.02,41.2,44.05,46.63
XS GIS Cut Line= 6
-609544.89559999   -1045215.8779-609568.07849999   -1045159.3655
-609569.86809999   -1045139.4457    -609584.1468   -1045094.0638
-609585.04899999   -1045083.2359-609645.95609999   -1044969.5427
#Sta/Elev= 30
       0  365.85    13.5   364.9   16.02  363.51   24.53  362.37   32.97  357.44
   43.75   356.7   51.15  356.45   51.73  355.95   52.11  356.46   54.11  356.24
   64.97  356.19   66.77  356.21   67.81  353.69   70.12  353.36   74.01  353.46
   75.45  353.71   77.54   356.2   112.1   356.1  127.58  356.28  133.49  356.79
  133.91  356.12   135.2  356.12  135.36  356.53   135.7     357  143.17  356.27
  152.93  356.95  211.03  356.88  228.34  357.09  241.83  357.04   268.5  371.35
#Mann= 3 ,-1 , 0
       0     .15       0   64.97    .045       0   77.54     .15       0
Bank Sta=66.77,77.54
XS Rating Curve= 0 ,0
Exp/Cntr=0.3,0.1

Type RM Length L Ch R = 1 ,17602.02,44.99,45.33,43.77
XS GIS Cut Line= 4
    -609628.5299    -1045233.445-609649.70439999   -1045183.4506
    -609659.3708   -1045165.9417    -609730.4928    -1045017.789
#Sta/Elev= 30
       0  361.93     3.5  361.52    7.37  361.35   13.18   357.8   14.71  356.68
   33.99  355.14   58.85  354.85   60.79  352.48   67.79  352.73   68.56  355.16
   68.63  355.51   68.66355.5085   75.39  355.51   76.07  355.26   76.69   354.8
   77.19  355.22  102.87  355.11  128.03  355.87  169.26  355.83  184.11  356.08
   202.6  355.93  212.73  356.31   215.2  356.99  217.47   356.8  218.32  355.81
  219.64  355.81  220.85   357.1  224.09  357.36  230.35  360.47  238.63  364.94
#Mann= 3 ,-1 , 0
       0     .15       0   58.85     .04       0   68.66     .15       0
#Block Obstruct= 1 ,-1
   44.03   54.82357.9499
Bank Sta=58.85,68.63
XS Rating Curve= 0 ,0
Exp/Cntr=0.3,0.1

Type RM Length L Ch R = 1 ,17514.01,2.8,2.8,2.82
BEGIN DESCRIPTION:
17708  PF 227 ŽELEZNÝ MOSTEK V KVASINÁCH (F39)
END DESCRIPTION:
XS GIS Cut Line= 4
    -609698.4602   -1045261.8683     -609725.443   -1045231.8903
-609730.18059999   -1045212.4594-609799.52079999   -1045040.7983
#Sta/Elev= 30
       0  360.74   13.45  359.62   17.99  356.01   19.82  355.95   20.92  354.22
   42.05  354.32   45.47     355   47.45354.6392   47.81  352.09   48.83  351.72
   53.33  351.94   56.51  352.88   56.63  354.56   56.64   354.7   66.87  354.91
   74.05  354.08  108.73  354.29  128.22  355.11  154.53  354.58  168.29  355.23
  198.31  355.56  214.27  355.33  214.89  354.69  215.58  355.14  220.87  355.47
  223.59  356.93  226.48  356.46  227.14  355.57  228.65  355.57  245.47  364.99
#Mann= 3 ,-1 , 0
       0     .15       0   47.45     .04       0   56.63     .15       0
Levee=-1,45.03,354.64,-1,67.26,354.77,,
#Block Obstruct= 2 ,-1
   87.04   98.39357.2969   24.15   30.84357.4231
Bank Sta=47.45,56.64
XS Rating Curve= 0 ,0
Exp/Cntr=0.5,0.3

Type RM Length L Ch R = 1 ,17511.2 ,12.67,11.2,9.7
XS GIS Cut Line= 4
    -609701.1935   -1045262.4972-609728.17619999   -1045232.5193
-609732.91389999   -1045213.0884-609802.25409999   -1045041.4272
#Sta/Elev= 30
       0  360.67   11.61  359.75   17.21  355.79   18.74  355.74   19.88  354.22
   41.62  354.21   45.47     355   47.44  354.71   47.83  351.43   48.13  351.32
   53.04  351.69    56.5  352.85   56.64   354.7   61.45  354.49   66.63  354.89
   74.68  354.08  106.42  354.22  127.47  355.01  155.19  354.56  196.68  355.45
  212.48   355.3  212.49  354.98  213.78  354.89  215.01  355.32  220.24  355.33
  223.38  356.66  225.83  356.46   226.4  355.57  227.98  355.57  245.47  365.11
#Mann= 3 , 0 , 0
       0     .15       0   47.44     .04       0   56.64     .15       0
Levee=-1,45.03,354.7,-1,65.82,354.72,,
#Block Obstruct= 3 ,-1
   86.57   97.92357.2387  145.42  164.87357.8016   18.01   30.73358.0956
Bank Sta=47.44,56.64
XS Rating Curve= 0 ,0
Exp/Cntr=0.5,0.3

Type RM Length L Ch R = 1 ,17440.04,41.3,46.93,51.33
XS GIS Cut Line= 4
-609760.83949999    -1045326.651-609797.06219999   -1045248.2126
    -609803.9891   -1045215.1089    -609864.0548   -1045079.3023
#Sta/Elev= 29
       0  357.96   25.55   358.3   31.64  355.71   35.65  353.91   45.53  353.87
   57.03  353.52   66.93  353.77   89.06  353.62  103.17  353.11   103.2  352.94
  104.02  350.75  110.53  350.85  112.14  353.96  120.22   353.9  121.54  353.76
  147.61  353.53  159.11  353.67     172  354.09  184.58   354.4  239.73  354.43
  240.01  354.29  245.36  353.92  251.56  354.58  254.38  356.22  257.06  356.15
  257.65  355.59   259.2  355.59  261.12   356.6  268.72  361.06
#Mann= 3 , 0 , 0
       0     .15       0  103.17     .04       0  112.14     .15       0
Levee=-1,66.86,353.76,-1,119.86,353.89,,
#XS Ineff= 2 , 0
           93.01  355.01  125.06          356.08
Permanent Ineff=
       F       F
#Block Obstruct= 4 ,-1
       0   17.78361.0793  182.05  227.99357.3547  138.13  160.15356.6496
   91.36  102.14356.3394
Bank Sta=103.17,112.14
XS Rating Curve= 0 ,0
Exp/Cntr=0.3,0.1

Type RM Length L Ch R = 1 ,17393.11,13.26,15.1,14.97
XS GIS Cut Line= 5
    -609773.9127   -1045343.0054    -609816.9842   -1045291.5139
-609843.09259999   -1045243.5518-609853.51619999   -1045227.0443
    -609891.0705   -1045107.7374
#Sta/Elev= 30
       0   357.3    4.31  355.16   28.77  355.07   35.81  355.35   38.43  354.22
   52.76  353.59   67.02  353.62   83.96   353.1   97.17  353.33  102.89  353.12
  117.97  353.22  123.95   352.8   126.5  350.88  132.18  350.89  132.74  352.01
  132.96  353.19  160.85  353.79  182.01  353.81  183.61  354.08  226.35  354.59
  242.41  354.53  248.19  354.04   251.2   354.3  256.76   354.1  257.29  353.76
   259.3  354.27  261.37  354.34  263.58  356.12  264.05  355.92  266.34     356
#Mann= 3 , 0 , 0
       0     .15       0  123.95     .04       0  132.96     .15       0
Levee=-1,67.02,353.62,0,,,,
#XS Ineff= 2 , 0
            96.6  354.06
Permanent Ineff=
       F       F
#Block Obstruct= 2 ,-1
   52.09    52.9356.6096   67.13    78.1356.4224
Bank Sta=123.95,132.96
XS Rating Curve= 0 ,0
Exp/Cntr=0.3,0.1

Type RM Length L Ch R = 1 ,17378   ,2.96,2.99,2.78
XS GIS Cut Line= 6
     -609777.842   -1045343.8274-609812.85159999     -1045322.95
    -609833.5683   -1045281.9181    -609866.1356    -1045237.247
    -609898.0165   -1045115.3894    -609907.0396   -1045097.3429
#Sta/Elev= 30
       0  356.33    4.12  355.13   40.29   354.5   59.87  353.74   93.02  353.51
   96.51  353.21   99.77  353.47  118.31  353.47  127.69  353.97  128.16  353.84
  128.17  353.23  128.18  351.66  132.69  350.83  135.79  351.67  135.87  353.64
  136.03  353.99   151.3  353.38  175.95  353.43  192.67  353.57  193.59  353.99
  195.42  354.03  247.07  354.26  263.29  353.47  267.08  354.21  269.69  355.94
  271.77  356.02  272.35  355.51  273.92  355.51  280.14  359.06  288.57  364.44
#Mann= 3 , 0 , 0
       0     .15       0  127.69     .04       0  136.03     .15       0
Levee=-1,127,353.97,-1,202.48,354.04,,
#XS Ineff= 2 , 0
                           144.8          355.87
Permanent Ineff=
       F       F
#Block Obstruct= 4 ,-1
   164.3  174.89356.4578  180.57  187.88356.5107   217.5   225.9357.2125
  236.65  247.52357.2125
Bank Sta=127.69,136.03
XS Rating Curve= 0 ,0
Exp/Cntr=0.5,0.3

Type RM Length L Ch R = 1 ,17375.01,8.74,9.01,9.67
XS GIS Cut Line= 6
    -609780.0582   -1045345.8438    -609815.0678   -1045324.9665
-609835.78449999   -1045283.9345-609868.35179999   -1045239.2635
    -609900.2327   -1045117.4058     -609909.256   -1045099.3593
#Sta/Elev= 30
       0  356.66    1.51  356.22     3.8  353.94   13.71  354.17   20.31   353.8
   42.47  353.75   45.33  354.19   54.28  353.43   87.05  353.15   94.83  352.77
   101.2  353.43  113.33  353.34  128.45  353.89  128.49  352.43   128.5  351.65
  133.03  350.82  136.13  351.64   136.2  353.67  136.27  353.94  152.01  353.35
  194.94  353.56  195.97  354.01  248.13  354.18  263.75  353.46  267.91  354.19
  270.65  355.98  272.83  356.06  273.43  355.51  275.01  355.51  288.57  363.86
#Mann= 3 , 0 , 0
       0      .1       0  128.45     .04       0  136.27      .1       0
Levee=-1,123.15,353.68,-1,140.13,353.75,,
#Block Obstruct= 3 ,-1
  165.99  176.58 356.446  182.19   189.5356.5049  218.36  248.38357.1706
Bank Sta=128.45,136.27
XS Rating Curve= 0 ,0
Exp/Cntr=0.5,0.3

Type RM Length L Ch R = 1 ,17366   ,28.61,25.35,19.86
XS GIS Cut Line= 5
    -609829.4397   -1045357.2129    -609861.4726   -1045259.9622
    -609876.1358   -1045246.3611    -609880.4211   -1045229.0826
    -609907.8099   -1045124.7443
#Sta/Elev= 30
       0  365.52   12.38  355.09   21.35  353.94   23.66  353.65    37.8  353.23
    61.6   352.8    72.7  352.91   79.98  353.14   80.52  353.26   80.93  352.56
   82.58   352.5    82.9  353.53    83.5   353.6   89.54  353.39   101.6  352.66
  106.24  352.26  108.13  351.52  111.97  350.79  116.19  351.52  116.56  353.71
   122.6  353.39  139.25   353.2  154.31   353.4  182.83  353.52  184.41  354.03
  217.23  354.12  232.88  354.01  244.41  353.58   245.3  353.44  248.07  353.81
#Mann= 3 , 0 , 0
       0      .1       0   101.6    .035       0  116.56      .1       0
Levee=-1,83.57,353.57,-1,118.79,353.57,,
#Block Obstruct= 3 ,-1
   65.59   77.29355.9429  224.73  231.42357.0443  121.07  132.79 356.422
Bank Sta=101.6,116.56
XS Rating Curve= 0 ,0
Exp/Cntr=0.3,0.1

Type RM Length L Ch R = 1 ,17340.65,22.16,21.68,21.33
XS GIS Cut Line= 2
    -609858.6317   -1045358.2556    -609920.0152   -1045174.1052
#Sta/Elev= 30
       0   364.4    9.97  354.97    15.3  354.18   17.56  352.73   24.41  352.86
   34.21  352.76   35.44  353.47   42.65  353.54   43.48  352.83   44.98  352.77
   62.04  352.76   76.22  353.29      85   353.1   86.18  353.89   87.07   353.9
   87.83   353.9   89.06  353.05   90.41  352.74   90.52  350.95   93.96   350.7
   98.72  351.52   98.92  353.29  100.25  352.88  110.89  352.81  151.11  353.26
  167.41  353.31  181.44  353.15  187.01  353.46  189.85  354.24  194.11  354.12
#Mann= 3 , 0 , 0
       0      .1       0   90.41    .037       0   98.92     .15       0
Levee=-1,86.84,353.75,-1,99.42,353.11,,
#Block Obstruct= 3 ,-1
  104.51  123.54355.8673   47.65   49.81355.7874  160.17   161.2356.2895
Bank Sta=90.41,98.92
XS Rating Curve= 0 ,0
Exp/Cntr=0.3,0.1

Type RM Length L Ch R = 1 ,17318.97,27.08,26.98,26.72
XS GIS Cut Line= 2
    -609884.2434   -1045362.2772    -609936.7369   -1045178.5502
#Sta/Elev= 30
       0  363.16    6.23   359.1   12.51  354.79   15.36  354.65   16.89  353.64
   18.51   352.4   21.88  352.37   32.69  352.62    42.4  352.39   49.01  352.37
   50.32     353   58.54  353.08   72.71  352.92   81.96  353.08   83.21  353.62
   84.33  353.65   86.16  352.48   87.18  352.44   87.38  350.54   93.44  350.84
   94.66  352.66  121.45  352.65  131.72  352.98  143.99  353.08  153.18  353.39
  168.15  353.21  185.65  353.31  186.95  353.38  189.85  354.18  191.08  354.15
#Mann= 3 , 0 , 0
       0      .1       0   87.18    .045       0   94.66      .1       0
Levee=-1,83.6,353.22,0,,,,
#Block Obstruct= 3 ,-1
   55.63   72.46355.9849  152.78  162.47356.3312  112.64  123.92355.7037
Bank Sta=87.18,94.66
XS Rating Curve= 0 ,0
Exp/Cntr=0.3,0.1

Type RM Length L Ch R = 1 ,17199.2 ,15.17,16.71,17.13
XS GIS Cut Line= 4
-609970.81529999   -1045391.2756-610024.34479999    -1045305.958
    -610027.6521   -1045292.7288-610079.25149999   -1045167.8199
#Sta/Elev= 30
       0  359.33    2.01  359.33    5.47  356.75   10.93  356.22   16.16  351.95
   28.98  351.45   32.98   351.4   46.06  351.56   66.39  351.52    93.4  351.68
  104.68  351.48  106.49  349.62  106.73  349.61  112.17  349.74  114.08  351.32
  114.43  351.42  135.27  351.89  146.56  351.88  149.72  351.77  194.77  351.83
  195.14  351.64  197.92  351.65  200.02  351.94  202.05   351.6  213.74  351.47
  234.32  351.48  235.01  350.86  236.43  350.85  243.28   354.1   249.5  355.35
#Mann= 3 , 0 , 0
       0      .1       0  104.68     .05       0  114.43      .1       0
Levee=0,,,-1,135.25,351.89,,
#XS Ineff= 1 ,-1
   60.05   92.96  354.04
Permanent Ineff=
       F
#Block Obstruct= 2 ,-1
   51.48   65.97354.5328   95.54  104.67354.5594
Bank Sta=104.68,114.43
XS Rating Curve= 0 ,0
Exp/Cntr=0.3,0.1

Type RM Length L Ch R = 1 ,17182.49,12.56,21.69,26.56
XS GIS Cut Line= 4
-609984.94399999   -1045394.1508-610038.65459999   -1045311.8652
    -610045.5337   -1045293.3443    -610102.7465   -1045177.3449
#Sta/Elev= 30
       0  357.41    4.11  356.92    8.48  352.44    9.38  351.63   16.51  351.08
    35.6  350.98   36.46   351.4   61.86  351.38   77.25  351.62   92.75  351.72
  104.98  351.53  107.02  349.78  111.16  349.53  113.38  349.57  115.02  351.23
  118.76  351.34  128.15  351.26   128.7  351.32  129.24  351.68  155.18  351.75
  171.85  352.01  189.49  351.91   191.3  351.29  222.11  351.26  228.44  351.52
  229.27  350.86  230.26  350.86   230.7  351.14  231.06  351.69  247.36  352.99
#Mann= 3 , 0 , 0
       0      .1       0  104.98     .05       0  115.02     .09       0
Levee=0,,,-1,172.78,351.92,,
#XS Ineff= 1 ,-1
   37.53   81.12   352.8
Permanent Ineff=
       F
#Block Obstruct= 4 ,-1
   82.86   92.82354.6667    8.03   15.49355.0234   48.72   71.72354.4726
  170.04  180.75354.9718
Bank Sta=104.98,115.02
XS Rating Curve= 0 ,0
Exp/Cntr=0.3,0.1

Type RM Length L Ch R = 1 ,17145.99,27.89,32.71,30.59
XS GIS Cut Line= 4
-609997.46979999   -1045397.9022-610062.86769999   -1045325.5206
    -610080.0049   -1045315.2094    -610182.7567   -1045191.3149
#Sta/Elev= 30
       0  357.24    6.15  351.67    14.1     351   24.39  350.83   32.11  351.25
   37.64   351.3   91.97  351.04   97.39  350.99   99.35  350.81  104.81  349.89
  105.71  349.55  110.73  349.04  112.06   349.9  113.36  351.14  113.98  351.29
  122.05  351.09  124.36  351.43  141.11  351.03  199.41  350.88  208.51  350.64
  221.71  350.56  222.39  349.96  223.87  349.96  224.34  350.56  227.21  350.67
  265.19  351.15  266.17  351.32  269.86   353.2  272.83  354.95  278.51  358.84
#Mann= 3 , 0 , 0
       0      .1       0   99.35     .05       0  113.98      .1       0
Levee=0,,,-1,114.15,351.27,,
#XS Ineff= 1 ,-1
   32.39   68.76  352.71
Permanent Ineff=
       F
#Block Obstruct= 2 ,-1
  144.81  157.32 354.041    3.59   11.11355.6489
Bank Sta=99.35,113.98
XS Rating Curve= 0 ,0
Exp/Cntr=0.3,0.1

Type RM Length L Ch R = 1 ,17072.46,16.25,12.79,10.07
XS GIS Cut Line= 3
    -610056.4079   -1045446.8883    -610113.0288   -1045371.7464
-610223.62489999   -1045234.1628
#Sta/Elev= 30
       0  362.86    5.81  362.76   11.04  357.35   17.41  350.27   26.76  350.11
   36.49  350.63   75.89  350.41   76.02  350.41   77.72  348.61   85.07  348.96
   86.69  350.19  115.69  349.61  117.06  350.65  124.26  350.78  125.58  350.24
  141.31  350.71  160.37  350.85  203.33  350.69  208.96  350.51  217.84  350.63
  220.67  350.45  239.18  350.25  240.04  349.23  241.23  349.23  242.23  350.24
  253.12  350.86  255.34  351.26  261.63  353.52  263.12  354.36  270.61  359.31
#Mann= 3 , 0 , 0
       0      .1       0   75.89     .05       0   86.69     .08       0
Levee=0,,,-1,124.23,350.77,,
#Block Obstruct= 1 ,-1
   15.82    28.3354.4257
Bank Sta=75.89,86.69
XS Rating Curve= 0 ,0
Exp/Cntr=0.3,0.1

Type RM Length L Ch R = 1 ,16981.23,7.15,8.37,7.3
XS GIS Cut Line= 5
    -610135.9278   -1045473.8311-610172.04879999   -1045435.4654
    -610183.2412   -1045429.7737-610209.17089999   -1045395.1544
    -610278.8182   -1045285.8913
#Sta/Elev= 30
       0  359.36    2.91  356.09    8.22  350.74    8.61   349.8   17.89   349.6
   25.37  349.59   27.28  349.73   35.71  349.56   53.52  349.57   56.11   348.1
   59.56  347.77   62.22  347.94   63.57   348.2   63.58  350.14   70.75  349.99
   76.88  350.18   77.52  350.37   84.05  350.07   84.83  349.82   108.5  350.02
  126.53  349.86  144.31   350.1  162.23  349.82  197.73  349.84  224.27  349.52
  225.05  348.85  226.58  348.85  232.02  350.74  235.04  352.34  238.08  354.11
#Mann= 3 , 0 , 0
       0     .09       0   53.52    .045       0   63.58      .1       0
Levee=0,,,-1,77.51,350.34,,
#Block Obstruct= 2 ,-1
  109.64  133.82352.9926   10.37   21.53352.6887
Bank Sta=53.52,63.58
XS Rating Curve= 0 ,0
Exp/Cntr=0.3,0.1

Type RM Length L Ch R = 1 ,16972.87,6.4,7.07,5.77
XS GIS Cut Line= 4
-610141.14319999    -1045476.769-610175.05779999   -1045443.1728
    -610187.6253   -1045437.0179    -610283.7571   -1045290.0894
#Sta/Elev= 30
       0  360.27    8.52  351.82    9.48  349.63   19.56  349.52   27.77  349.69
   39.38  349.58   49.32  349.81   52.24  347.83   55.24  347.66   58.72  348.06
   59.08  348.59   59.09  350.16    59.6  350.18   59.65  350.16   59.72  349.93
   60.78   349.9   74.43  350.15   76.38  350.31   83.13  349.95   83.39  349.85
  131.46  349.79   147.6  350.02  165.87  349.79  193.69   349.8  209.31  349.57
  225.93  349.46  226.67  348.85  228.32  348.85  231.83  350.98  237.31  353.65
#Mann= 3 , 0 , 0
       0     .08       0   49.32    .045       0   59.09      .1       0
Levee=0,,,-1,76.48,350.29,,
#Block Obstruct= 3 ,-1
   65.48   72.46353.0419  109.79  133.97352.8312   12.12   23.49 352.596
Bank Sta=49.32,59.09
XS Rating Curve= 0 ,0
Exp/Cntr=0.3,0.1

Type RM Length L Ch R = 1 ,16947.94,14.61,14.1,13.66
XS GIS Cut Line= 6
    -610169.5517   -1045485.6161-610173.24989999    -1045477.427
    -610183.6554   -1045466.7471-610201.92269999   -1045457.7056
    -610218.8174   -1045438.1758    -610302.8072   -1045298.9794
#Sta/Elev= 30
       0  356.32    4.38  352.23    6.07  350.95    6.77  350.22   19.78  349.49
   22.82  349.66    23.9  349.91   28.73  349.91   28.74  348.84   29.13  348.41
   30.46  347.61   37.39  347.77   38.04  348.04   40.11  349.42   48.72  349.64
   59.87  349.69   61.96  349.79   64.59  350.12   76.11  349.83  109.33  349.71
  119.86  349.78  172.83  349.51  185.94  349.61  197.09  349.42   222.4  349.38
  222.92   348.8   224.5   348.8  227.52  350.97  228.79  352.13  232.67  354.58
#Mann= 3 , 0 , 0
       0      .1       0   28.73    .045       0   40.11     .09       0
Levee=0,,,-1,64.52,350.09,,
#XS Ineff= 2 , 0
           25.69  350.98
Permanent Ineff=
       F       F
Bank Sta=28.73,40.11
XS Rating Curve= 0 ,0
Exp/Cntr=0.3,0.1

Type RM Length L Ch R = 1 ,16933.84,27.14,24.89,15.43
XS GIS Cut Line= 6
    -610172.8312   -1045503.2958    -610183.6262   -1045487.4208
    -610192.1378   -1045478.4949    -610208.3665   -1045469.9668
    -610228.7441   -1045448.1827    -610312.5439   -1045301.5194
#Sta/Elev= 30
       0  364.96    6.16   364.6    8.34  362.41   19.24  349.88   21.81   349.6
   31.53  350.04   32.63  349.98   36.25  347.68   43.98  347.81    44.6  348.34
    46.6  349.24   47.05  349.28      74  349.63   76.83     350   82.89  349.84
    88.8  349.51   99.14  349.54  105.83  349.75  137.71  349.66  141.24  349.75
  173.25  349.39  218.78  349.42  227.56  349.21  235.14  349.26  235.67  348.69
  237.01  348.69  239.77  351.08  241.66  352.51   246.9  355.87  248.61  356.83
#Mann= 3 , 0 , 0
       0      .1       0   32.63     .05       0   47.05      .1       0
Levee=0,,,-1,76.79,349.93,,
#XS Ineff= 2 , 0
           29.73   351.8
Permanent Ineff=
       F       F
#Block Obstruct= 2 ,-1
   54.52   58.56352.4616   62.43   72.37352.5712
Bank Sta=32.63,47.05
XS Rating Curve= 0 ,0
Exp/Cntr=0.3,0.1

Type RM Length L Ch R = 1 ,16908.96,23.54,18.95,17.48
XS GIS Cut Line= 4
    -610198.8204   -1045514.3025-610207.27569999   -1045500.8694
-610218.91739999    -1045490.286-610326.86769999   -1045304.5481
#Sta/Elev= 30
       0  364.82    1.92  364.81    5.06  361.73   15.76  349.93   16.33  350.09
   20.47  349.69   23.63  347.55   27.25  347.55   32.28  347.77   32.56  348.01
   35.84  348.99   45.46  349.24   58.51  349.32   74.81  349.61   83.76  349.44
   89.85  349.43  140.81  349.74  149.89  349.63   155.7  349.46  171.89  349.47
  173.96  349.35  178.22  349.47  197.19  349.33  211.07  349.38  227.15  349.19
  228.01  348.62  229.58  348.88  231.73  350.63  238.74  355.68  246.44  359.96
#Mann= 3 , 0 , 0
       0      .1       0   20.47     .05       0   35.84      .1       0
Levee=0,,,-1,74.62,349.53,,
Bank Sta=20.47,35.84
XS Rating Curve= 0 ,0
Exp/Cntr=0.3,0.1

Type RM Length L Ch R = 1 ,16890.01,24.27,25.01,24.32
XS GIS Cut Line= 4
-610221.34499999   -1045523.4945-610227.91319999   -1045511.4527
    -610232.1466   -1045500.3402-610348.03429999    -1045310.369
#Sta/Elev= 30
       0  363.81    2.72  363.71    12.3  349.23   15.89  349.05   16.62  348.91
   18.76  347.34   28.64  347.64   32.41  348.84   78.95  349.52  154.27  349.65
  165.49     350  166.92     350  167.77  349.53  176.48  349.33  177.43   349.5
  180.22  349.17  186.76  349.28  191.62  350.27  195.13  349.24  198.05  349.07
   205.7  349.29  217.16  349.34     218  349.19  219.11   349.8  220.63  350.19
   225.7   350.4  228.92  352.03  230.56  352.65  240.37  359.02  248.14  362.93
#Mann= 3 , 0 , 0
       0      .1       0   15.89     .05       0   32.41      .1       0
Levee=0,,,-1,79.1,349.54,,
Bank Sta=15.89,32.41
XS Rating Curve= 0 ,0
Exp/Cntr=0.3,0.1

Type RM Length L Ch R = 1 ,16865   ,23.67,25.02,24.87
XS GIS Cut Line= 4
    -610242.3339   -1045535.2969-610251.72569999   -1045518.8611
-610256.48829999   -1045506.6902-610363.90929999   -1045327.8315
#Sta/Elev= 30
       0  362.48    3.55  362.51    8.65  357.25   15.13  350.15   15.97  349.86
   16.89  349.05    20.4  348.03   21.45  347.14   24.84  347.03   30.54  347.08
    33.6  348.75   75.61  349.48  125.31  349.12  172.22  349.86  174.95   349.2
  178.82  350.81  180.57  351.01  183.03  350.95  186.06   350.3  189.92  350.01
  192.38  348.89  193.39  348.82  200.93  348.65  216.51  348.91  217.48  349.33
  218.28  349.22  218.88  348.57  221.31  349.05  224.02  349.96  240.64  358.73
#Mann= 3 , 0 , 0
       0      .1       0   16.89     .05       0    33.6      .1       0
Levee=0,,,-1,73.04,349.36,,
#Block Obstruct= 3 ,-1
   40.16   42.34351.8377   53.17   61.37352.1396  124.09  141.85352.2846
Bank Sta=16.89,33.6
XS Rating Curve= 0 ,0
Exp/Cntr=0.3,0.1

Type RM Length L Ch R = 1 ,16839.98,20.16,18.86,18.8
XS GIS Cut Line= 5
    -610259.1032   -1045553.0799-610271.81769999   -1045531.5794
    -610281.7151      -1045514.2-610303.42729999   -1045472.5025
-610381.65659999   -1045334.2117
#Sta/Elev= 30
       0  362.01   11.21  361.43    26.6  348.95   27.07  348.62   31.89  347.45
   32.73  346.87   35.66  346.79   38.62  346.82    40.2  348.45   50.96  348.39
   83.99  349.08   93.27   349.1    94.6  348.62  117.31  349.35  130.81  348.81
  130.81  348.56  137.38  348.59   166.5  349.56  167.74  349.22  198.45  348.46
  204.51  348.72   205.7  349.26  208.22   349.8  213.87  348.79  224.12  348.86
  226.41  349.59  229.39  350.15  229.96  349.35  233.32  349.68  250.87     360
#Mann= 3 , 0 , 0
       0      .1       0    26.6     .05       0    40.2      .1       0
Levee=0,,,-1,87.12,349.06,,
#Block Obstruct= 3 ,-1
   45.64   52.53351.4954     131  148.77351.7318   95.79   114.2 351.951
Bank Sta=26.6,40.2
XS Rating Curve= 0 ,0
Exp/Cntr=0.3,0.1

Type RM Length L Ch R = 1 ,16821.12,43.01,41.79,41.65
XS GIS Cut Line= 2
-610275.27459999   -1045565.3143    -610395.3498   -1045343.0538
#Sta/Elev= 30
       0  361.46    3.71  360.82    6.05  360.65   17.33  360.98   20.94  358.62
   29.19  350.56   32.12   349.4   34.27  348.04   34.85  346.74   38.31  346.66
   41.55  346.67   43.58  348.44   54.15  348.27   66.86   348.4   93.44  349.04
  108.69  349.14  142.41  348.97  161.72  349.11  168.37  349.38   169.6  348.98
  171.36  348.92  202.82  348.56  212.54  348.64  214.81  348.83  229.46  348.84
  232.68  349.89   235.9  350.15  236.56  349.58  242.45  352.12  252.62  359.44
#Mann= 3 , 0 , 0
       0      .1       0   32.12     .05       0   43.58     .05       0
Levee=0,,,-1,167.67,349.28,,
#Block Obstruct= 1 ,-1
   53.58   64.61351.3344
Bank Sta=32.12,43.58
XS Rating Curve= 0 ,0
Exp/Cntr=0.3,0.1

Type RM Length L Ch R = 1 ,16779.33,27.37,27.39,27.36
XS GIS Cut Line= 3
-610308.17929999   -1045592.8645    -610344.1895   -1045525.2731
    -610422.3832   -1045375.8722
#Sta/Elev= 30
       0  360.74   13.01   359.7   27.24  359.17   30.05  359.24   31.05  356.79
   35.49  356.79   41.52   349.1   41.67  348.96   41.68  348.82   42.18  346.88
   42.35  346.77    46.1  346.58   50.53  346.71   51.68  348.04   52.23  348.16
   55.08  348.35   62.56  348.37   68.18  348.25   88.19  348.39   99.57  348.61
  144.02  348.74  156.41  349.05   172.7  348.67  210.75  348.47  223.51   348.6
  238.02  348.97  239.52  349.94  243.06  349.94  243.51  349.69  245.21   349.7
#Mann= 3 , 0 , 0
       0      .1       0   41.52     .05       0   52.23      .1       0
Levee=0,,,-1,157.04,349.04,,
#Block Obstruct= 4 ,-1
   54.68   61.27351.3319  145.23  155.83351.9062  111.15  121.79351.6265
    20.1   29.15362.3344
Bank Sta=41.52,52.23
XS Rating Curve= 0 ,0
Exp/Cntr=0.3,0.1

Type RM Length L Ch R = 1 ,16751.94,21.77,21.42,20.49
XS GIS Cut Line= 3
-610331.99179999   -1045606.3583     -610368.002   -1045538.7669
    -610450.4891    -1045381.048
#Sta/Elev= 30
       0  359.83    3.86  359.16    7.68  358.91    13.1  358.87   13.71  358.77
   21.76  358.45   26.44  358.34   26.69  358.03   36.22     352   37.03  351.14
    39.3   349.4    43.3  346.47   46.95  346.38   51.43  346.62   53.67  347.82
   55.59  347.96   63.34  348.27    84.5   348.4  103.36  348.42  119.61  348.07
  137.55  348.17  154.31  348.46  188.11   348.8   214.3  348.57  232.32  348.69
   236.5  348.74  249.53  349.21  250.98  349.63  251.15  350.05  254.57  349.95
#Mann= 3 , 0 , 0
       0      .1       0    39.3     .05       0   55.59      .1       0
#XS Ineff= 2 , 0
                          104.45          351.53
Permanent Ineff=
       F       F
#Block Obstruct= 2 ,-1
  184.93  199.08351.7553   56.68   63.33351.1675
Bank Sta=39.3,55.59
XS Rating Curve= 0 ,0
Exp/Cntr=0.3,0.1

Type RM Length L Ch R = 1 ,16730.52,4.86,4.82,4.85
XS GIS Cut Line= 3
    -610352.6812   -1045617.9347-610388.15709999   -1045543.0952
    -610465.3939   -1045389.8634
#Sta/Elev= 30
       0  358.93    9.19  357.93   14.08  358.21   22.01  357.45   27.93  354.09
   32.64  353.17   38.18  349.89   42.75  348.86   43.07   348.4   43.43   346.9
   44.17  346.39   48.14  346.29   52.25  346.36   53.34  346.67   53.78  347.08
   55.17  347.83   55.91  348.02   68.85  348.23    86.3  347.93   97.54  348.18
  109.47  347.99  131.38  347.96  142.98  348.11   148.1  348.02  181.48  348.75
  216.45  348.58  235.97  348.67  252.59  348.92  253.94  350.02  254.42  350.01
#Mann= 3 , 0 , 0
       0      .1       0   42.75     .05       0   55.91      .1       0
Levee=0,,,-1,182.74,348.68,,
#XS Ineff= 2 , 0
                          113.87          352.02
Permanent Ineff=
       F       F
#Block Obstruct= 2 ,-1
   58.22   64.91351.0959       0    8.43361.4715
Bank Sta=42.75,55.91
XS Rating Curve= 0 ,0
Exp/Cntr=0.5,0.3
